HEC-RAS study SECONDCK.prj: SECONDCK

--- SECONDCK.g01 (geometry) --- (continued)

Type RM Length L Ch R = 1 ,83139   ,504.7,492.6,481.8
XS GIS Cut Line= 4
     2135636.417      211853.076     2135888.386      212115.768
     2136079.684      212313.848     2136433.569      212384.344
#Sta/Elev= 30
       0 2320.93      23 2319.71      59 2315.36      82 2301.58   108.2 2292.81
   127.9  2289.7   137.7 2284.15   147.6 2282.64   167.2 2286.68   229.6 2284.68
   239.4 2285.69   268.9 2282.92   288.6 2284.69   308.2 2284.62   318.1 2283.16
   350.9 2283.41   373.8 2282.85   380.4 2283.86   393.5 2286.55   432.8 2284.88
   462.4 2285.79   570.5 2284.06   596.8 2287.15   639.4 2298.52   721.4 2326.92
   737.8 2334.33   757.5 2337.36   767.3  2343.5   780.4 2349.13  1000.2 2426.19
#Mann= 9 ,-1 , 0
       0    .035       0     110     .07       0   350.9    .045       0
   380.4     .07       0     394      .1       0     494     .07       0
     544      .1       0  669.37     .04       0  869.37      .1       0
Bank Sta=350.9,380.4
XS Rating Curve= 0 ,0
Exp/Cntr=0.3,0.1

Type RM Length L Ch R = 1 ,82646   ,534,549.6,542.8
XS GIS Cut Line= 4
     2135154.923      212032.781     2135173.152       212225.49
2135834.60870281212615.8770975172136429.16623273212592.556690927
#Sta/Elev= 30
       0 2335.75    53.9 2325.32    73.7 2320.27   109.9 2309.51   146.2 2294.43
   179.1 2287.01   278.1 2285.11   297.2 2281.83   312.4 2283.78   468.6 2282.66
   514.3 2283.51   565.5 2282.53   583.6 2280.71   605.8 2279.68     6262280.628
   636.5 2282.54   722.6 2282.49   735.3  2281.4   758.5 2282.72   817.2 2282.84
   849.7 2280.19   868.6 2283.49    1246 2283.16    1268 2284.73  1309.1 2295.97
  1377.3  2337.8    1397 2340.17  1410.1  2347.4  1498.6 2378.52  1556.7 2395.04
#Mann= 8 ,-1 , 0
       0    .035       0   583.6    .045       0     626    .035       0
  943.57     .06       0 1141.64    .035       0 1301.64      .1       0
 1341.64     .04       0 1431.64      .1       0
#XS Ineff= 2 , 0
                         1099.62         2341.73
Permanent Ineff=
       F       F
Bank Sta=583.6,626
XS Rating Curve= 0 ,0
Exp/Cntr=0.3,0.1

Type RM Length L Ch R = 1 ,82097   ,515.9,515.6,449.1
XS GIS Cut Line= 3
  2134625.244012212312.2493666342135618.46692828212852.603802952
2136395.54807003212801.141475683
#Sta/Elev= 30
       0 2316.03    30.6 2314.93    80.7 2305.79   158.1 2295.62   235.5  2290.3
   494.4 2285.02   559.7 2281.38   628.2 2281.72   639.5 2280.24   663.8 2280.04
     815 2281.18   852.5  2280.1   874.7 2281.04   886.2 2279.86   893.7 2277.78
     908 2277.63   919.6 2276.83     927 2277.51   938.2 2280.15  1005.5 2281.88
  1651.7 2282.34  1697.8 2281.41  1753.7 2293.29  1781.4 2304.58  1809.1 2317.54
  1855.6 2336.12  1867.7 2339.24  1888.5 2341.22  1901.6    2349  1909.5 2352.08
#Mann= 12 ,-1 , 0
       0     .06       0     200     .04       0     230     .06       0
     350     .04       0     410     .06       0     460    .035       0
     820     .07       0     908    .045       0     927     .06       0
  1430.7     .07       0  1720.7    .035       0  1820.7     .04       0
#XS Ineff= 2 , 0
                            1400         2286.01
Permanent Ineff=
       F       F
Bank Sta=908,927
XS Rating Curve= 0 ,0
Exp/Cntr(USF)=0,0
Exp/Cntr=0.3,0.1

Type RM Length L Ch R = 1 ,81581   ,641.7,637.7,546.2
XS GIS Cut Line= 2
      2134232.18       213167.33     2136437.041      212885.212
#Sta/Elev= 30
       0 2337.33    72.1 2324.84   265.6 2304.84     282 2300.04   311.5 2300.34
   383.6 2290.85     459 2284.84   504.9 2282.79   609.8 2281.35   806.5 2280.63
   885.2 2278.22     895 2276.86   934.4 2278.48   957.3 2276.27   980.3 2278.76
  1009.8 2279.11  1026.2 2276.66  1055.7 2278.55  1121.2 2279.47  1137.6 2276.86
  1150.8 2276.57  1183.6 2278.61  1209.8 2277.57  1232.7 2280.18  1291.7 2280.59
  1721.2 2281.89  1980.2 2280.67  2003.2 2283.78  2081.9 2315.22  2222.8 2351.59
#Mann= 13 ,-1 , 0
       0    .035       0     500     .07       0   934.4    .045       0
   980.3     .07       0    1200    .035       0    1300     .06       0
    1500     .07       0    1600     .04       0    1700     .06       0
    1790     .07       0    1990    .035       0    2090      .1       0
    2130     .04       0
#XS Ineff= 2 , 0
                         1562.07         2285.28
Permanent Ineff=
       F       F
Bank Sta=934.4,980.3
XS Rating Curve= 0 ,0
Exp/Cntr=0.3,0.1

Type RM Length L Ch R = 1 ,80943   ,533.5,528.6,515.4
XS GIS Cut Line= 2
2134434.83340111213748.048297421 2136447.0103973212909.212362947
#Sta/Elev= 30
       0 2336.75    47.1 2333.94   114.8 2327.16   224.8 2313.47   263.9 2306.98
   306.5 2305.14   374.1  2299.2   385.6 2297.62   395.6 2294.05   420.3 2295.47
   452.3  2292.2     516 2281.08   541.1 2278.48   637.1 2276.52   709.2 2278.51
   932.1 2278.19  1165.8 2276.36  1178.3 2274.96  1184.5 2274.27  1208.72275.073
  1223.2 2278.01    1348 2279.25  1696.4 2280.88  1938.1  2279.7  1970.1 2282.75
  2016.3 2302.56  2041.7  2311.4  2108.7 2327.03  2122.9 2332.43    2180 2347.28
#Mann= 13 ,-1 , 0
       0    .035       0     680     .07       0     750    .035       0
    1070     .07       0  1178.3    .045       0  1208.7     .06       0
    1280     .07       0    1600     .06       0    1820     .07       0
    1920      .1       0    1960    .035       0    2030      .1       0
    2140     .04       0
#XS Ineff= 2 , 0
                         1368.42         2281.33
Permanent Ineff=
       F       F
Bank Sta=1178.3,1208.7
XS Rating Curve= 0 ,0
Exp/Cntr(USF)=0,0
Exp/Cntr=0.3,0.1

Type RM Length L Ch R = 1 ,80415   ,938.7,929.3,893.3
XS GIS Cut Line= 2
     2134753.013       214261.08     2136441.381      212928.615
#Sta/Elev= 30
       0  2365.3    45.9 2363.18    98.4 2354.86   180.3 2337.06   311.5 2317.99
   350.8 2309.26     377 2307.88   396.7 2303.72   413.1 2303.46     518 2280.12
     600 2277.23   721.3 2277.26   757.4 2275.17   944.3 2276.22   960.7 2274.08
   973.8 2272.41   983.6 2274.14    1000 2276.37  1068.9 2274.56  1091.8 2276.81
  1160.7  2276.8  1213.1 2278.58  1275.4 2277.73    1777 2280.19  1888.5 2279.05
  1944.3 2282.08  1973.8 2284.43  2029.5    2307  2095.1 2323.39  2150.8 2340.94
#Mann= 13 ,-1 , 0
       0    .035       0     600     .07       0     620    .035       0
     730     .07       0     780    .035       0     850     .07       0
   960.7    .045       0   983.6     .07       0    1090    .035       0
    1410     .07       0    1850    .035       0    1890      .1       0
    2100     .04       0
#XS Ineff= 2 , 0
                         1257.88            2305
Permanent Ineff=
       F       F
Bank Sta=960.7,983.6
XS Rating Curve= 0 ,0
Exp/Cntr=0.3,0.1

Type RM Length L Ch R = 1 ,79485   ,346.1,347.3,346.4
XS GIS Cut Line= 2
2135109.26115051214715.1445062152136555.92435039213062.631997264
#Sta/Elev= 30
       0 2310.49    46.3 2309.86    83.9 2304.11   118.4 2302.57   187.7 2303.01
   245.2 2295.86   323.7 2293.31   345.5 2289.47   360.2  2289.5   371.9 2291.34
   464.8 2285.34   586.1 2279.83     626 2276.42   804.2 2274.25  838.57  2271.4
   851.3 2270.98   890.5 2271.48   929.8 2273.93  1014.5 2275.43  1218.7 2275.21
    1283 2277.08  1534.3 2278.46  1694.7 2277.51  1711.8 2278.72  1894.7 2279.99
  1915.6 2281.55  2085.3  2305.6  2111.4 2306.94  2159.7 2315.68  2196.3 2325.92
#Mann= 7 ,-1 , 0
       0    .035       0  838.57    .045       0   890.5    .035       0
    1370     .07       0    1900    .035       0    2030      .1       0
    2160     .04       0
Bank Sta=838.57,890.5
XS Rating Curve= 0 ,0
Exp/Cntr(USF)=0,0
Exp/Cntr=0.3,0.1

Type RM Length L Ch R = 1 ,79138   ,833,849.1,834
XS GIS Cut Line= 3
     2135447.458      214855.698     2136636.694      213471.149
     2136701.798      213254.136
#Sta/Elev= 30
       0 2304.35    85.2 2299.64     118 2295.82   199.9  2293.6   242.5 2288.66
   301.5 2278.99   350.6 2275.98   704.5 2274.23   714.3 2271.49   730.7 2271.72
   740.6  2274.3   865.1 2272.95   914.2 2273.63   969.9 2271.65   996.1 2273.31
    1160 2274.76  1346.8 2275.87  1356.6    2275  1513.9 2278.18  1599.1  2282.6
  1782.6 2295.43  1815.3 2295.34  1825.2 2297.31  1851.1 2299.35    1864 2297.87
  1902.8 2303.16  1941.7 2311.14  1970.8  2319.9  2012.9 2329.32  2051.7 2342.01
#Mann= 8 ,-1 , 0
       0    .035       0   704.5    .045       0   740.6    .035       0
    1160     .07       0    1320    .035       0    1420     .07       0
    1550    .035       0 1915.17      .1       0
#XS Ineff= 2 , 0
                         1235.92         2276.79
Permanent Ineff=
       F       F
Bank Sta=704.5,740.6
XS Rating Curve= 0 ,0
Exp/Cntr=0.3,0.1

Type RM Length L Ch R = 1 ,78289   ,1065,1084.9,1025.4
XS GIS Cut Line= 2
2135906.65596098215158.1160645752137033.68092816213871.557882865
#Sta/Elev= 30
       0 2313.37    62.5 2303.24   123.2 2295.06   152.5 2285.32   174.1 2284.75
   202.3 2275.23   217.2 2273.01   327.5  2272.1   369.4 2270.36   441.3 2272.52
   568.1 2272.56   578.6 2269.72   592.6 2269.42   622.8 2269.87   635.5 2273.41
   768.7 2273.68   786.2 2271.43   799.3 2273.07   909.3 2274.39   939.2 2272.99
     965 2274.85     994 2272.97  1056.6 2275.18  1094.8 2274.61  1352.4 2278.86
    1423 2283.12    1484 2291.45  1575.6 2300.46  1645.4 2303.95  1710.4 2309.86
#Mann= 7 ,-1 , 0
       0     .04       0     160    .035       0     260     .04       0
   578.6    .045       0   622.8    .035       0    1440      .1       0
    1500    .035       0
#XS Ineff= 2 , 0
                          852.63         2276.57
Permanent Ineff=
       F       F
Bank Sta=578.6,622.8
XS Rating Curve= 0 ,0
Exp/Cntr(USF)=0,0
Exp/Cntr=0.3,0.1

Type RM Length L Ch R = 1 ,77204   ,1388,1412.8,1361.9
XS GIS Cut Line= 2
     2136280.791      215341.809     2137365.861      214191.636
#Sta/Elev= 30
       0  2318.9    36.1 2296.49    75.4 2274.63    95.1 2273.62   108.3  2270.8
   223.1 2270.11   242.8 2269.24   262.4 2271.39   278.8 2269.04   321.5 2271.23
   459.3 2271.77   488.8 2270.35     538  2272.2   626.6  2270.8   744.7 2270.71
   751.2 2269.58   764.4  2268.2  775.05 2269.58     807 2272.45   905.4 2272.56
  1082.6 2277.64  1105.6 2279.05  1154.8 2279.36  1269.6 2283.64  1328.6 2287.98
  1381.1 2289.31  1394.2 2291.73    1427 2295.05  1538.6 2302.59  1581.2 2306.49
#Mann= 13 ,-1 , 0
       0    .035       0     180     .04       0     390    .035       0
     470     .04       0     520    .035       0     610     .04       0
   751.2    .045       0  775.05     .04       0     790    .035       0
    1040     .04       0    1180      .1       0    1330    .035       0
    1470     .04       0
#XS Ineff= 2 , 0
                          810.53         2274.15
Permanent Ineff=
       F       F
Bank Sta=751.2,775.05
XS Rating Curve= 0 ,0
Exp/Cntr=0.3,0.1

Type RM Length L Ch R = 1 ,75791   ,982.9,1004.2,984.4
XS GIS Cut Line= 2
      2136732.18      215949.448     2137752.145      214847.018
#Sta/Elev= 30
       0 2324.47    16.4 2317.03    68.9 2290.12    88.5 2282.01   111.5 2274.69
   124.6 2269.22   147.6 2269.35   157.4 2265.53   160.7 2265.33   183.6 2267.72
   432.9 2267.88   452.5 2269.05   495.2  2267.2   521.4 2265.65   531.2  2267.6
   541.1 2269.17   593.5 2268.13   629.6 2269.23     810 2269.34   960.8 2269.08
   993.6 2270.65  1006.7 2269.82    1151 2269.62  1259.2 2271.88  1295.3 2274.54
  1370.7 2282.74  1380.6  2285.6    1397 2287.28  1436.3 2294.95  1501.9 2309.08
#Mann= 10 ,-1 , 0
       0      .1       0     140    .035       0     240     .04       0
     410    .035       0   495.2    .045       0   531.2    .035       0
     810     .04       0    1110    .035       0    1350     .04       0
    1400      .1       0
#XS Ineff= 2 , 0
                          989.47         2272.56
Permanent Ineff=
       F       F
Bank Sta=495.2,531.2
XS Rating Curve= 0 ,0
Exp/Cntr=0.3,0.1

Type RM Length L Ch R = 1 ,74787   ,469.5,474,464.7
XS GIS Cut Line= 2
2136874.14771363216151.3389808542138129.82849898215477.182493639
#Sta/Elev= 30
       0 2325.05    16.3 2318.35    62.3 2288.06    99.6  2268.7   103.5 2267.52
   125.6  2267.8   139.9 2263.83   185.9 2266.93   237.3 2267.85   360.2 2267.62
   409.1 2265.64   436.9 2268.08   479.4 2267.36     498 2265.41   524.1 2266.32
   546.4 2265.07   576.2 2267.99  732.99 2265.81   743.2 2264.71   750.4 2265.79
   762.4 2267.19   806.2    2267     822 2268.73  1273.8  2276.6  1310.1 2280.95
  1322.2 2284.05  1335.9 2284.35    1373  2293.4  1404.6 2303.88  1425.2 2308.67
#Mann= 10 ,-1 , 0
       0      .1       0      30    .035       0     250     .04       0
     470    .035       0  732.99    .045       0   750.4    .035       0
     920     .04       0    1060    .035       0    1140     .04       0
    1260    .035       0
#XS Ineff= 2 , 0
                          823.16          2274.4
Permanent Ineff=
       F       F
Bank Sta=732.99,750.4
XS Rating Curve= 0 ,0
Exp/Cntr(USF)=0,0
Exp/Cntr=0.3,0.1

Type RM Length L Ch R = 1 ,74313   ,405.4,408.2,387.6
XS GIS Cut Line= 3
     2136897.111      216261.948     2137122.805       216287.99
     2138242.597      215940.768
#Sta/Elev= 30
       0 2332.46    35.7  2325.6    71.4 2316.24    97.4 2304.15     159 2269.06
   162.3 2267.75     185 2267.15     198 2263.46   217.5 2266.25   400.8 2266.81
   453.2 2264.98   476.1 2266.86   495.7 2267.21   505.6 2266.07   521.9 2267.58
     571 2266.49     594 2267.79   607.1 2267.32   620.2 2265.09   626.7 2263.38
   643.1 2263.52   649.6 2265.48     702 2265.28   721.7 2264.04   734.8 2266.84
   777.4  2267.2   800.3 2268.72   993.5 2270.92  1271.9 2279.44  1399.6 2281.65
#Mann= 7 ,-1 , 0
       0      .1       0     100    .035       0  377.19     .04       0
  407.19    .035       0   620.2    .045       0   649.6    .035       0
  917.19     .04       0
Bank Sta=620.2,649.6
XS Rating Curve= 0 ,0
Exp/Cntr=0.3,0.1

Type RM Length L Ch R = 1 ,73905   ,590.7,599.3,581.6
XS GIS Cut Line= 2
 2136933.1975115216727.8062114972138349.34909575216017.724538938
#Sta/Elev= 30
       0 2342.12    42.6 2335.02    65.1  2330.2    83.5 2322.42   108.6 2313.62
   159.9 2289.92   196.6 2277.81   211.9 2270.39   215.6 2269.39   235.7 2268.77
   243.1 2266.97   252.3 2263.19   263.3 2265.85     278 2266.62   313.9 2265.69
   663.3 2263.95   685.8 2265.21   727.72264.884   736.8 2262.07   746.6  2261.9
   755.1 2262.21   763.62264.943   865.2 2266.59   879.9 2265.31  1095.7 2269.73
  1269.7 2271.69  1357.7 2275.05  1503.8 2278.36  1541.1 2280.92  1584.2 2285.78
#Mann= 6 ,-1 , 0
       0      .1       0     180    .035       0     400     .04       0
   727.7    .045       0   763.6    .035       0     950     .04       0
Bank Sta=727.7,763.6
XS Rating Curve= 0 ,0
Exp/Cntr(USF)=0,0
Exp/Cntr=0.3,0.1

Type RM Length L Ch R = 1 ,73305   ,200.4,198.8,197.7
XS GIS Cut Line= 2
 2137223.9426115217099.1228749922138663.12181651216377.332692663
#Sta/Elev= 30
       0 2357.63    56.2 2348.65   101.5 2336.43   156.5 2308.76   196.6 2285.56
   220.7 2274.12     228 2269.32   231.7 2268.12     250 2267.81   266.4 2262.37
   284.5  2264.6   334.9 2264.78   514.3 2264.38   555.2 2263.08   628.4 2264.35
   657.82262.204   668.4 2260.26   686.8 2259.92     6972261.921   706.4 2264.33
   734.5 2262.61   955.7  2264.4   980.2 2264.13   991.4 2262.44  1126.1 2262.58
  1199.2 2265.76  1527.3 2270.26    1579 2272.24  1593.7 2275.65    1610 2275.91
#Mann= 7 ,-1 , 0
       0      .1       0     300    .035       0     370     .04       0
     590    .035       0   657.8    .045       0     697    .035       0
     850     .04       0
Bank Sta=657.8,697
XS Rating Curve= 0 ,0
Exp/Cntr(USF)=0,0
Exp/Cntr=0.5,0.3

Type RM Length L Ch R = 1 ,73107   ,66.8,66.3,66.1
XS GIS Cut Line= 4
      2137170.94      217511.318     2137743.465      217072.712
     2138045.548      216892.156     2138757.354      216531.045
#Sta/Elev= 30
       0 2342.16    88.4 2338.35   141.7 2333.05   187.1 2324.19   211.9 2316.53
   236.7 2306.56   282.2 2300.18   290.4 2297.52   310.7  2293.8   335.9 2288.43
     369 2279.32     402 2268.07   414.4 2264.83   477.5 2265.28   504.5  2264.8
   520.6 2263.08   743.3 2262.45   857.9 2264.29   877.62261.851   888.5 2259.82
   913.52261.936   982.3 2263.37  1132.2 2263.12  1318.5 2264.91  1383.4  2266.9
  1506.1  2266.5  1796.8 2270.02  1848.3 2272.02    1863 2276.84  1871.3 2277.46
#Mann= 8 ,-1 , 0
       0      .1       0   282.2    .035       0   310.7      .1       0
     402    .035       0   520.6     .04       0   877.6    .045       0
   913.5    .035       0  1132.2     .04       0
#XS Ineff= 5 ,-1
       0     700    2275     700     850    2275     920    1070    2275
    1070    1370    2275    1370  1871.3    2275
Permanent Ineff=
       F       F       F       F       F
Bank Sta=877.6,913.5
XS Rating Curve= 0 ,0
Exp/Cntr=0.5,0.3

Type RM Length L Ch R = 1 ,73040   ,199.8,206.1,199
XS GIS Cut Line= 4
     2137163.996      217601.596      2137767.77      217135.212
     2138069.854      216954.656     2138781.659      216593.545
#Sta/Elev= 30
       0 2318.65    22.3 2320.48    63.8 2319.61   118.2 2316.76     167 2312.11
   188.9 2308.19   223.2 2299.41   291.8 2279.17   345.7 2267.92   387.2 2266.97
   410.3 2263.62   424.5 2262.19     450 2262.34   532.3 2262.42   883.1 2262.56
   894.3 2264.92   921.4 2262.31   928.5 2259.85   936.3 2259.66   959.6 2259.86
   966.7 2262.28   971.6 2263.09  1024.3 2260.74  1043.5 2261.14  1054.8 2263.81
  1062.1 2263.99  1185.9 2263.03  1454.5 2264.56  1621.3 2266.65    1913 2274.87
#Mann= 9 ,-1 , 0
       0      .1       0   291.8    .035       0   410.3     .04       0
     450    .035       0   532.3     .04       0   894.3    .035       0
   921.4    .045       0   966.7    .035       0  1185.9     .04       0
#XS Ineff= 4 ,-1
       0  695.11  2268.5  695.11  848.412268.886  997.43    11102268.945
    1110    1722    2269
Permanent Ineff=
       F       F       F       F
Bank Sta=921.4,966.7
XS Rating Curve= 0 ,0
Exp/Cntr=0.5,0.3

Type RM Length L Ch R = 1 ,72834   ,667.6,691.8,677.3
XS GIS Cut Line= 2
2137162.24964505217701.1631874112138858.93956829216665.058516996
#Sta/Elev= 30
       0 2292.79    30.5 2295.46    77.9 2296.18   115.7 2294.44   168.8 2286.99
   230.4 2271.22     238 2268.22   245.7 2267.67   272.6 2267.33   299.5  2263.2
   417.8  2261.9   587.8 2261.94   701.1 2261.89   841.6 2259.99   974.5 2263.17
  1014.6 2263.79  1029.4 2262.09  1038.9 2259.67  1068.4 2259.69  1081.7 2262.02
  1122.2 2263.63  1148.1 2261.66  1185.8 2263.41  1410.5 2263.22  1713.6 2267.19
  1914.1 2272.01  1937.2 2272.94  1956.4  2276.4  1979.5 2275.32    1988 2276.72
#Mann= 9 ,-1 , 0
       0      .1       0   245.7    .035       0   417.8     .04       0
   587.8    .035       0   701.1     .04       0   974.5    .035       0
  1029.4    .045       0  1081.7    .035       0  1410.5     .04       0
#XS Ineff= 2 , 0
          513.13 2268.64 1355.56         2268.04
Permanent Ineff=
       F       F
Bank Sta=1029.4,1081.7
XS Rating Curve= 0 ,0
Exp/Cntr(USF)=0,0
Exp/Cntr=0.3,0.1

Type RM Length L Ch R = 1 ,72152   ,623.1,627.8,610.5
XS GIS Cut Line= 3
2137206.33797291217856.1223345072137585.72116359217642.934092852
2139375.65630167216934.239129826
#Sta/Elev= 30
       0 2269.89    99.7 2269.04   152.4 2265.02   202.6 2263.52   464.2 2261.71
   481.9 2261.43     492 2259.86   504.6 2261.01   628.5 2262.01     679 2261.42
   699.4 2259.59   745.2 2261.98   829.8 2262.04     846 2259.66   857.1 2258.81
   872.2 2259.58   882.8 2262.54   893.4 2262.79  1073.4 2261.87  1122.7 2259.87
  1133.3 2261.15  1182.1 2261.96    1430 2261.46  1538.5 2262.68  1972.8 2263.23
  2041.5 2264.75  2050.8 2268.65    2079 2269.15  2269.5 2294.97  2360.3 2301.66
#Mann= 8 ,-1 , 0
       0     .04       0    99.7    .035       0   202.6     .04       0
     846    .045       0   872.2    .035       0  1073.4     .04       0
  1972.8    .035       0  2050.8     .04       0
#XS Ineff= 2 , 0
          755.05 2268.05 1063.13         2268.19
Permanent Ineff=
       F       F
Bank Sta=846,872.2
XS Rating Curve= 0 ,0
Exp/Cntr(USF)=0,0
Exp/Cntr=0.3,0.1

Type RM Length L Ch R = 1 ,71524   ,636.9,659.2,647.4
XS GIS Cut Line= 2
     2137316.774      218362.013 2139585.4730327216944.428785468
#Sta/Elev= 30
       0 2281.66   168.1  2269.1   225.3 2262.54   252.6 2261.07   386.2 2262.79
   401.2 2261.14   498.4 2260.64   512.6 2258.37   527.7 2260.74   785.1 2260.61
   822.9  2259.4     862 2260.85   873.6 2258.51   885.2 2256.98   896.8 2258.95
   906.2 2260.35   939.8 2259.85   954.9 2261.25  1214.1 2258.91  1461.7 2260.86
  2113.4 2262.14    2161 2264.15  2185.1 2268.27  2208.3  2267.8  2222.9 2271.46
    2330 2282.85  2432.7 2295.07  2498.5 2298.95  2579.7 2299.08  2675.2 2293.32
#Mann= 10 ,-1 , 0
       0    .035       0     470     .04       0   873.6    .045       0
   896.8     .04       0     900    .035       0    1360     .04       0
    2180    .035       0    2290     .04       0    2330    .035       0
    2410     .04       0
#XS Ineff= 2 , 0
             619 2262.75 1809.56         2262.75
Permanent Ineff=
       F       F
Bank Sta=873.6,896.8
XS Rating Curve= 0 ,0
Exp/Cntr=0.3,0.1

Type RM Length L Ch R = 1 ,70865   ,728.1,752.3,718.7
XS GIS Cut Line= 3
2137246.37143755218472.6880165992139216.77165193217927.909501314
2140122.37749551217340.680712111
#Sta/Elev= 30
       0 2287.34    79.2 2278.68   208.6 2272.85   309.3  2261.6   604.8 2260.61
   767.5 2260.03   786.2 2257.52   802.2 2260.16   933.6 2258.55   977.9 2260.23
  1236.6 2259.62  1301.3 2257.53  1314.2 2256.09  1323.9 2257.51    1383    2260
  1439.5 2259.33  1457.8 2258.01  1508.6 2260.52  1545.5 2258.47  1566.8 2260.22
  2445.2  2265.4  2462.3  2269.1  2477.2 2269.06  2493.1 2266.47    2575 2268.66
  2825.1  2273.2  2889.2  2273.4  2911.2 2270.03  2955.6 2274.94  3123.7    2279
#Mann= 9 ,-1 , 0
       0    .035       0   604.8     .04       0  1301.3    .045       0
  1323.9    .035       0  1439.5     .04       0    2575    .035       0
  2825.1     .04       0  2889.2    .035       0  2911.2     .04       0
Bank Sta=1301.3,1323.9
XS Rating Curve= 0 ,0
Exp/Cntr(USF)=0,0
Exp/Cntr=0.3,0.1

Type RM Length L Ch R = 1 ,70113   ,944.4,959.4,955.8
XS GIS Cut Line= 3
     2137474.368      218705.5242139678.84454975218564.922129741
2140088.77738542218945.028454513
#Sta/Elev= 30
       0  2289.6   117.7 2278.83   193.3 2264.47   249.2 2258.39   459.6 2258.89
   541.7 2256.01   574.6 2258.19   617.4 2257.04   702.8 2258.51   722.6 2255.31
   735.7 2257.81   778.4 2258.46   794.9 2256.15     799 2253.38     808 2252.51
   821.2 2253.09     831 2256.44   850.8 2258.04   900.1 2254.86   919.8 2258.52
   937.3 2258.93  1015.1 2259.12  1039.3 2255.79  1057.9 2258.29  1107.1 2259.25
  2390.5  2264.6  2432.3 2268.06  2443.9 2271.24  2562.9 2277.93    2768 2302.56
#Mann= 5 ,-1 , 0
       0    .035       0   794.9    .045       0     831     .08       0
    1100    .035       0    1200     .04       0
#XS Ineff= 2 , 0
                         1212.12         2266.99
Permanent Ineff=
       F       F
Bank Sta=794.9,831
XS Rating Curve= 0 ,0
Exp/Cntr=0.3,0.1

Type RM Length L Ch R = 1 ,69153   ,614.3,618.4,610.2
XS GIS Cut Line= 2
      2137504.75      218983.302     2139217.815      219587.707
#Sta/Elev= 30
       0 2287.63   127.9 2274.73   137.7 2272.06   167.2 2260.51   190.2 2257.56
     400 2257.42   455.8 2257.25   468.9 2254.81   485.3 2255.46   498.4    2254
   524.6 2256.64   609.9  2255.9   615.9 2253.54     623 2250.95   632.8 2251.15
   642.7 2253.84   659.1 2253.04   672.2 2256.06   685.3  2256.7   836.1  2257.1
   862.4 2261.39   885.3 2268.72     905 2269.43   921.4  2269.1   944.4 2263.82
    1587 2263.85  1626.4 2268.47  1642.8 2268.94  1780.5 2269.03  1816.6 2266.73
#Mann= 12 ,-1 , 0
       0     .04       0      60    .035       0     400     .08       0
     610     .07       0   615.9    .045       0   642.7     .07       0
     650      .1       0     820     .08       0     920      .1       0
     940    .035       0    1030    .025       0    1650    .035       0
Bank Sta=615.9,642.7
XS Rating Curve= 0 ,0
Exp/Cntr=0.3,0.1

Type RM Length L Ch R = 1 ,68535   ,641.7,628.6,599.2
XS GIS Cut Line= 2
2137311.57749541 219343.958839932138855.44731346219889.459508975
#Sta/Elev= 30
       0  2271.4      78 2273.95   133.6 2272.91   171.9 2270.57   234.6  2264.7
   265.6 2259.69   293.9 2258.17   314.5 2258.64   356.3 2256.22     371 2257.25
   394.6 2255.91   516.4 2255.97   596.4 2254.08   655.6 2255.53   686.9 2252.57
   700.1 2254.26   721.7 2254.14     749 2253.36   764.4 2251.39   780.8 2249.63
   788.3 2251.22   798.2  2256.5   895.9 2256.25  1000.1 2257.62  1017.5 2259.98
  1052.3 2268.18  1069.7 2269.14  1083.6 2268.72  1104.5 2263.83  1637.4 2263.82
#Mann= 11 ,-1 , 0
       0    .035       0     290     .07       0     400     .08       0
     500     .07       0     610     .08       0     750      .1       0
   764.4    .045       0   788.3      .1       0    1020     .08       0
    1040      .1       0    1130    .025       0
Bank Sta=764.4,788.3
XS Rating Curve= 0 ,0
Exp/Cntr(USF)=0,0
Exp/Cntr=0.3,0.1

Type RM Length L Ch R = 1 ,67906   ,490.5,492.2,479.6
XS GIS Cut Line= 2
     2137183.569      220120.455     2138841.555      219925.143
#Sta/Elev= 30
       0 2313.12   150.9 2282.88   206.6 2274.16   226.3 2272.01   255.8 2258.74
   265.7 2255.55   291.9  2254.1     410 2254.21   426.4 2255.03   528.1 2255.14
     551 2254.25   560.9 2249.63   580.5 2249.42   603.5 2253.94   619.9 2254.72
   698.6 2253.72   711.7 2251.71   728.1 2254.01     879 2254.34   924.9 2253.54
  1000.4  2255.5  1154.5 2257.11  1226.7 2256.62  1249.6 2257.32  1275.9 2259.57
  1302.1 2265.42  1321.8  2266.3  1331.6 2265.88  1344.7 2263.82  1669.4 2263.82
#Mann= 11 ,-1 , 0
       0     .04       0      10    .035       0     310      .1       0
     410     .08       0     551    .045       0   603.5     .08       0
     700      .1       0     900     .08       0    1100      .1       0
    1300     .03       0    1400    .025       0
Bank Sta=551,603.5
XS Rating Curve= 0 ,0
Exp/Cntr=0.3,0.1

Type RM Length L Ch R = 1 ,67414   ,745.9,754.4,756.8
XS GIS Cut Line= 3
2137244.67646996220568.7622289172138587.84321166220301.158127122
2139030.41922617220398.936548931
#Sta/Elev= 30
       0 2304.12    84.3 2299.75     274 2278.17   300.4 2271.67   313.8 2270.77
   342.8 2256.49   354.9 2253.05     568 2253.24   601.5 2250.79   614.9 2252.51
   641.6 2248.72   661.7  2252.2   728.6 2253.52     742 2249.96     752 2249.49
   762.1 2252.26   792.2 2252.66   805.5 2249.13     829 2249.61   840.12251.991
    1120 2257.18  1135.9 2259.85  1208.5 2261.18  1364.2 2261.97    1381 2260.11
  1411.2 2262.27  1646.7  2265.8  1730.4 2273.74  1771.7 2283.85  1822.8 2290.34
#Mann= 9 ,-1 , 0
       0     .04       0     350     .08       0     450      .1       0
     480     .08       0   792.2    .045       0   840.1     .08       0
     850      .1       0     980     .08       0    1150      .1       0
Bank Sta=792.2,840.1
XS Rating Curve= 0 ,0
Exp/Cntr(USF)=0,0
Exp/Cntr=0.3,0.1

Type RM Length L Ch R = 1 ,66660   ,629.6,650.1,610.3
XS GIS Cut Line= 2
2137301.92960441220858.5547805842138559.99237505220937.867433515
#Sta/Elev= 30
       0  2310.3   126.1 2303.55   188.5 2295.12     205 2291.53   218.1 2286.43
   231.3 2284.92   234.5 2283.29   241.1 2277.85   287.1 2251.86   298.62251.349
   310.2 2247.09   329.9 2246.74     343 2247.54   351.82251.431   398.9 2251.69
   431.9 2250.29   477.8 2251.34     629 2250.29   638.9    2253   648.2 2257.53
   694.8 2285.97   707.9 2287.66   717.8 2293.63   744.1 2300.04   800.3 2308.58
   826.3 2311.52   947.9 2319.12  1076.1 2330.99  1227.3 2340.79  1260.6 2341.35
#Mann= 4 ,-1 , 0
       0     .04       0     190      .1       0   298.6    .045       0
   351.8      .1       0
Bank Sta=298.6,351.8
XS Rating Curve= 0 ,0
Exp/Cntr(USF)=0,0
Exp/Cntr=0.3,0.1

Type RM Length L Ch R = 1 ,66010   ,397.7,442.6,462.6
XS GIS Cut Line= 3
     2137287.736      220914.726     2137457.006      221166.462
     2138155.791      221366.115
#Sta/Elev= 30
       0 2313.44    81.6  2310.5   163.1 2287.84   205.5 2277.99   228.3 2274.64
     274 2271.47   316.4 2264.61   329.5 2264.08   336.1  2261.3   349.2 2259.18
   368.8 2248.77   375.4 2246.85     395  2246.8   408.1 2250.21   421.2 2251.26
   486.7 2252.22   499.8 2247.39   509.6 2246.26   539.1 2247.35     562 2247.54
   578.3 2250.32   637.3 2248.79   683.1  2250.6   715.8 2258.71   755.1 2275.29
   768.2  2277.2   787.8 2284.79     837 2295.86   935.2 2308.87  1030.1 2312.33
#Mann= 4 ,-1 , 0
       0     .04       0      70      .1       0   499.8    .045       0
   539.1      .1       0
Bank Sta=499.8,539.1
XS Rating Curve= 0 ,0
Exp/Cntr=0.3,0.1

Type RM Length L Ch R = 1 ,65567   ,357.7,354.3,338.8
XS GIS Cut Line= 2
     2137287.736      220940.768     2137604.576      221891.288
#Sta/Elev= 30
       0 2313.55    32.7 2312.32    39.3 2311.15    58.9 2303.51     108 2287.58
   163.7    2271   189.9 2264.96   216.1 2262.26   288.1 2258.48   389.6 2256.38
   422.4 2256.69   455.1  2254.7   497.7 2249.59   523.9 2249.78   540.3 2246.02
   546.8 2244.97   563.2 2244.88   582.8 2245.04   589.4 2246.76   602.5 2249.08
   638.5  2248.3   658.1 2252.94   710.5 2260.16   723.6  2265.6   743.3 2271.41
   795.7 2283.47   867.7 2308.56   897.2 2317.15   959.4 2329.38  1001.9 2336.36
#Mann= 4 ,-1 , 0
       0     .04       0      30      .1       0   540.3    .045       0
   589.4      .1       0
Bank Sta=540.3,589.4
XS Rating Curve= 0 ,0
Exp/Cntr=0.3,0.1

Type RM Length L Ch R = 1 ,65213   ,451.7,454.2,444.7
XS GIS Cut Line= 2
     2136784.263      221049.274     2137465.687      221908.649
#Sta/Elev= 30
       0  2335.6    19.6 2335.57    42.6 2333.49    58.9 2328.22    85.1 2313.49
   104.8 2299.46   121.1 2285.79     131 2275.47   150.6 2259.86     167  2250.8
   176.8 2248.11   428.9 2249.68   523.8 2251.79   546.7 2250.27   563.1 2245.11
   599.1 2243.84   612.2 2244.86   628.6 2246.18     645 2251.55   667.9 2255.74
   687.5 2257.42   766.1 2258.16   779.2 2260.09   798.8 2265.79   844.7 2271.25
   910.1 2287.56  1005.1 2300.66  1018.2 2304.12  1070.6 2323.83  1096.8 2331.08
#Mann= 3 ,-1 , 0
       0      .1       0   563.1    .045       0   612.2      .1       0
#XS Ineff= 2 , 0
          369.23 2300.33
Permanent Ineff=
       F       F
Bank Sta=563.1,612.2
XS Rating Curve= 0 ,0
Exp/Cntr=0.3,0.1

Type RM Length L Ch R = 1 ,64758   ,504.7,561.6,597.6
XS GIS Cut Line= 2
     2136545.548      221422.538     2137287.736       222073.58
#Sta/Elev= 30
       0 2284.84    49.2 2283.23    88.6 2278.21   144.3  2275.6   193.5  2279.9
   213.2 2280.54   252.6 2288.16   275.5 2290.86     305 2292.56     328  2291.9
   370.6 2286.96   400.2 2285.15   442.8  2278.1   465.8 2272.92   501.8  2262.9
   567.4 2253.78   593.7 2245.84   629.8 2243.29   646.2 2245.79   692.1 2247.21
   724.9 2245.19   741.3 2245.56   747.8  2244.6   774.1 2247.19   780.6 2249.44
   816.7 2268.09     843  2280.2   892.2 2300.43   938.1 2315.79   987.3 2339.38
#Mann= 3 ,-1 , 0
       0      .1       0   593.7    .045       0   646.2      .1       0
Bank Sta=593.7,646.2
XS Rating Curve= 0 ,0
Exp/Cntr=0.3,0.1

Type RM Length L Ch R = 1 ,64197   ,536.3,558.2,573.7
XS GIS Cut Line= 3
     2136523.847      221405.1772136651.68363781221717.256043935
     2136467.423      222203.788
#Sta/Elev= 30
       0 2283.88      59 2282.43   115.7 2277.29   203.5 2274.59   250.5 2271.27
   285.9 2267.64   314.3 2263.35   334.9 2258.82   350.7  2251.4   367.1 2248.49
   395.2 2247.64   419.8 2245.54   446.6 2247.33   464.4 2246.79   479.4 2247.58
   521.5 2245.36   546.1 2245.78   549.6  2245.3   560.1 2240.89   591.6 2240.25
   600.9 2241.58   605.7 2246.25   609.2 2251.03   612.7 2254.29   623.2 2260.53
   682.9 2290.26   702.7 2301.22   721.5 2309.99   802.8 2353.86   857.5 2382.25
#Mann= 3 ,-1 , 0
       0      .1       0   546.1    .045       0   605.7      .1       0
Bank Sta=546.1,605.7
XS Rating Curve= 0 ,0
Exp/Cntr=0.3,0.1

Type RM Length L Ch R = 1 ,63639   ,460.5,455.6,450.6
XS GIS Cut Line= 3
        2136411.      221353.094     2136108.021       221640.82
      2135852.96      221900.462
#Sta/Elev= 30
       0 2268.48    32.6 2265.09    84.9 2256.77   117.5 2249.44   130.6 2248.01
   189.3 2245.61     222 2245.53   251.4 2244.32   310.1 2244.15   326.4 2245.56
   339.5  2244.4   349.3  2241.4   352.5 2241.08   378.7 2240.34   388.4 2238.24
     408 2238.05   444.1 2238.37   450.6 2241.58   453.9 2243.64     467 2249.38
   499.8 2269.32     526 2282.93   562.1 2300.82   581.8 2308.33   614.6 2315.12
   670.3 2321.43   716.2 2322.19   729.3 2323.53     749 2324.05   781.8 2323.04
#Mann= 3 ,-1 , 0
       0      .1       0   378.7    .045       0   450.6      .1       0
Bank Sta=378.7,450.6
XS Rating Curve= 0 ,0
Exp/Cntr=0.3,0.1

Type RM Length L Ch R = 1 ,63183   ,375.6,335.5,304.7
XS GIS Cut Line= 3
     2136059.437      221005.872     2135764.298      221387.816
     2135807.701      221856.566
#Sta/Elev= 30
       0 2280.12      13 2273.83    39.1 2265.86    81.5  2256.3   120.7 2248.77
   208.7 2242.24   228.3  2241.5   251.1 2242.52   264.2 2241.37   277.2 2241.32
   280.5 2240.52   283.7 2238.79   290.3 2235.88   332.7 2235.67   342.4  2236.5
     349 2238.78   365.3 2242.42   375.1 2243.57   401.2 2242.85   446.8 2243.71
   476.2 2249.38   521.9 2251.57     571 2255.03   737.7 2272.69   809.6 2278.52
   822.7 2280.55   865.2 2290.62   933.8 2304.06   943.6 2305.31   953.4 2307.75
#Mann= 3 ,-1 , 0
       0      .1       0   283.7    .045       0     349      .1       0
Bank Sta=283.7,349
XS Rating Curve= 0 ,0
Exp/Cntr=0.3,0.1

Type RM Length L Ch R = 1 ,62848   ,312.4,307.7,300.7
XS GIS Cut Line= 3
2135575.94880495220927.1683135892135721.81115517221410.337348685
2135782.58713443221869.195992079
#Sta/Elev= 30
       0 2330.14     7.3 2327.72    17.8 2322.71    38.9 2307.63    52.6 2296.67
    63.4 2286.73   109.9 2249.99   121.1 2239.26   124.5 2237.31     131 2236.14
   151.7 2235.62   169.1 2235.91     181    2239   199.9 2241.85   213.6 2241.19
   223.9 2242.31   275.3 2243.44   322.7 2241.27     337  2242.1   364.4 2240.35
   391.8 2242.03   426.1  2242.1   494.3 2247.68     575 2252.43   706.8 2264.65
   786.2 2270.47   814.6 2273.53   855.5 2281.35   945.1 2301.93   967.6 2306.16
#Mann= 3 ,-1 , 0
       0      .1       0   121.1    .045       0     181      .1       0
Bank Sta=121.1,181
XS Rating Curve= 0 ,0
Exp/Cntr(USF)=0,0
Exp/Cntr=0.3,0.1

Type RM Length L Ch R = 1 ,62540   ,554,584.5,636
XS GIS Cut Line= 3
     2135498.197      220941.874     2135369.333      221205.524
     2135741.253      221892.395
#Sta/Elev= 30
       0 2326.82    58.7 2323.81    78.3 2321.91   146.7 2311.66   176.1 2304.91
   189.1 2301.46   277.2 2270.93   296.7 2259.88   306.5 2253.35   329.4  2243.5
   335.9 2238.48   342.5 2237.28   352.3 2243.02   358.8 2243.53   371.9 2237.42
   378.4 2234.94   388.2 2234.43   430.7 2234.58   443.8 2237.11   453.6 2238.85
     483 2238.59   522.2 2241.54   656.2 2241.21   741.2 2245.71   829.4 2252.57
   894.8 2260.07   973.2 2272.03   999.4 2279.15  1028.8 2288.71  1074.6 2300.99
#Mann= 3 ,-1 , 0
       0      .1       0   371.9    .045       0   443.8      .1       0
Bank Sta=371.9,443.8
XS Rating Curve= 0 ,0
Exp/Cntr=0.3,0.1

Type RM Length L Ch R = 1 ,61956   ,813,814.9,841.1
XS GIS Cut Line= 2
     2135450.454      220898.471     2134708.267      221866.353
#Sta/Elev= 30
       0  2323.5    75.4 2316.06   150.8 2301.82   196.7 2289.77   298.4  2253.3
   331.2 2246.43   373.8 2242.14   390.2 2236.47   413.1 2239.99   475.4 2240.11
   537.7 2237.07   734.4  2239.9   744.3 2238.55   750.8  2235.2   757.4 2232.05
   767.2 2231.66   793.4 2231.93   803.3 2235.35   829.5 2245.02   865.6 2252.78
   914.8 2266.94   934.4 2275.05   967.2 2292.53  1003.3 2306.52  1026.2 2316.92
  1039.4 2320.84  1052.5 2321.54  1127.9 2314.77  1190.2  2314.1  1219.7 2311.62
#Mann= 3 ,-1 , 0
       0      .1       0   750.8    .045       0   803.3      .1       0
Bank Sta=750.8,803.3
XS Rating Curve= 0 ,0
Exp/Cntr=0.3,0.1

Type RM Length L Ch R = 1 ,61141   ,524.9,529.3,527.4
XS GIS Cut Line= 3
     2135351.972      220745.455     2135176.024       220702.61
     2134569.378       221037.36
#Sta/Elev= 30
       0 2309.63   145.5 2298.82   190.9 2293.72     217 2288.72   223.6 2286.32
   230.1  2281.9   233.4  2278.2   243.2 2262.65   246.4 2259.99   282.4 2239.12
   298.8 2230.78   305.3 2228.54   311.8 2227.54   344.5 2227.37   347.8 2227.48
   354.3 2230.47   360.8 2233.26     387 2234.34   416.4    2234   452.4 2238.22
   462.2 2238.51   511.2 2246.64   547.1 2255.95   586.4 2269.04   602.7 2273.49
   681.1 2300.42   694.2 2301.34   733.4 2307.17   798.8 2314.64     874 2321.95
#Mann= 4 ,-1 , 0
       0      .1       0   298.8    .045       0   354.3      .1       0
  701.09    .035       0
Bank Sta=298.8,354.3
XS Rating Curve= 0 ,0
Exp/Cntr=0.3,0.1

Type RM Length L Ch R = 1 ,60611   ,496.1,494.4,492.3
XS GIS Cut Line= 2
2135190.38210553220103.2074740372134396.11110553220580.638474037
#Sta/Elev= 30
       0 2250.83      61  2245.1    70.6 2242.98    80.6  2245.2   103.5 2244.25
   130.4 2246.01   213.2 2254.65     249 2254.92   329.4 2249.13   388.6  2240.2
   463.4 2234.47   478.7 2230.24     5052228.694   520.8 2225.79   555.9 2225.57
   563.1 2226.53   572.12230.306   578.2 2233.09     589 2234.08   603.8 2233.17
   647.1  2237.1   677.7  2249.7   700.7 2256.94   712.2 2257.18   723.7 2260.25
   765.8 2262.86   786.4 2267.38   811.8 2267.84   842.3 2271.14   926.7 2282.51
#Mann= 7 ,-1 , 0
       0      .1       0     430    .035       0     505    .045       0
   572.1     .08       0     660    .035       0     730      .1       0
     890    .035       0
Bank Sta=505,572.1
XS Rating Curve= 0 ,0
Exp/Cntr=0.3,0.1

Type RM Length L Ch R = 1 ,60117   ,706.6,709.5,709.5
XS GIS Cut Line= 2
      2135317.25      219391.288     2134175.756      220163.858
#Sta/Elev= 30
       0 2250.63    91.7 2247.86     131 2243.62   258.6 2244.04   491.1 2237.76
   523.8 2234.47   543.5 2235.98     645 2234.71   658.1 2231.42   671.2 2234.59
   690.8 2231.78     717 2234.14   923.3  2233.5     956 2231.91   978.9 2233.21
   985.5 2231.62     992 2226.37   998.6 2224.25  1008.4 2224.12  1031.3 2224.35
  1037.9 2226.08    1051 2231.16    1087 2231.53  1109.9 2234.17    1123 2238.76
  1139.4 2240.86  1152.4 2247.06    1195 2259.48    1231 2267.41  1378.4 2285.91
#Mann= 8 ,-1 , 0
       0    .035       0     840     .07       0     890      .1       0
     950     .08       0     992    .045       0  1037.9     .08       0
    1060     .07       0    1070    .035       0
#XS Ineff= 2 , 0
          715.01 2259.11
Permanent Ineff=
       F       F
Bank Sta=992,1037.9
XS Rating Curve= 0 ,0
Exp/Cntr=0.3,0.1

Type RM Length L Ch R = 1 ,59407   ,544.2,540.5,536.8
XS GIS Cut Line= 3
       2135129.1      218723.645     2133906.659      219486.774
      2134075.93      220159.518
#Sta/Elev= 30
       0  2273.1   147.4 2251.23   229.3 2245.89   504.4 2236.15   756.6 2231.17
   913.8 2230.77   936.7 2227.38   962.9 2230.92  1051.3 2230.71  1090.6 2228.98
  1159.4 2230.71  1169.2  2229.1  1175.8 2225.39  1182.4 2223.67  1211.8 2223.51
  1218.4 2225.39  1224.9 2229.69    1238 2231.88  1329.7 2231.74  1339.6 2230.17
  1388.7 2232.48  1414.9  2239.4  1441.1  2250.4  1493.4 2259.14  1519.6 2261.26
  1712.7  2264.7  1755.2  2267.7  1886.1 2282.45  1997.4 2283.46  2134.8 2293.24
#Mann= 7 ,-1 , 0
       0      .1       0      10     .04       0     710    .035       0
  1175.8    .045       0  1218.4    .035       0 1651.09      .1       0
 1861.09    .035       0
#XS Ineff= 2 , 0
         1021.44 2248.98 1295.71         2247.96
Permanent Ineff=
       F       F
Bank Sta=1175.8,1218.4
XS Rating Curve= 0 ,0
Exp/Cntr=0.3,0.1

Type RM Length L Ch R = 1 ,58867   ,471.9,415.9,371.6
XS GIS Cut Line= 4
2134906.00239332218164.8731247192133873.81259284218949.734807238
2133701.02724119219183.3292314612134054.12230906220136.084017365
#Sta/Elev= 30
       0 2249.72    66.6 2248.61    93.7 2245.29   153.3 2246.34   590.9 2235.39
  1064.9 2228.92  1072.2  2225.7  1077.3 2223.55  1099.6 2223.17  1114.4 2223.72
  1118.3 2225.72  1137.1  2228.9  1250.4 2227.48  1295.7 2229.95  1514.4 2226.55
  1521.6 2224.77  1554.7 2227.71  1590.3 2235.48  1660.2 2236.02  1719.7  2238.9
  1772.2 2246.69  1807.2 2255.02  1849.2 2260.73  1992.6 2270.89  2038.1 2273.05
  2125.6 2271.71  2201.9 2273.57  2393.3 2287.33  2517.5 2288.07  2603.3  2292.5
#Mann= 7 ,-1 , 0
       0     .04       0     970    .035       0    1060     .07       0
  1072.2    .045       0  1118.3    .035       0 2237.25      .1       0
 2337.25    .035       0
Bank Sta=1072.2,1118.3
XS Rating Curve= 0 ,0
Exp/Cntr(USF)=0,0
Exp/Cntr=0.3,0.1

Type RM Length L Ch R = 1 ,58451   ,498.6,502.1,499.2
XS GIS Cut Line= 4
2133047.81825449217488.0498022452133867.42002417218937.580885113
2133664.17769979 219171.260479862134028.47090963220149.184507317
#Sta/Elev= 30
       0 2269.86     100 2252.24   254.2 2237.41     266 2233.57   277.3 2236.37
   771.1 2226.88    1295 2229.08  1317.6 2228.59  1340.6 2223.35  1352.1 2222.35
  1397.8 2223.69  1431.6 2227.18  1494.7 2226.28  1665.2 2229.38  1861.9 2227.16
  1894.4 2224.22  1933.8 2228.13  1969.2 2242.34  1981.7 2244.77  2004.7 2246.47
  2050.6 2244.75  2123.8 2246.98  2267.4 2263.82  2400.4 2274.51  2445.9 2276.78
  2547.5 2276.31  2645.5 2279.34  2823.5 2291.21  2939.6 2291.44  3018.5 2295.08
#Mann= 5 ,-1 , 0
       0    .035       0  1340.6    .045       0  1397.8    .035       0
  2634.9      .1       0  2744.9    .035       0
#XS Ineff= 2 , 0
         1296.85 2230.77 1671.49         2230.96
Permanent Ineff=
       F       F
Bank Sta=1340.6,1397.8
XS Rating Curve= 0 ,0
Exp/Cntr(USF)=0,0
Exp/Cntr=0.3,0.1

Type RM Length L Ch R = 1 ,57949   ,210.5,201.5,185.4
XS GIS Cut Line= 2
 2132602.9203093  217716.50728332134020.95148536  220151.1043472
#Sta/Elev= 30
       0 2240.95    83.3 2243.75   136.5 2243.33   216.2 2244.95   292.2 2241.17
   436.4 2236.43   469.2 2234.25     534 2226.37   554.1 2225.46   755.4  2225.3
  1001.3 2223.16    1192 2224.46  1294.6 2223.05  1328.7 2224.34  1336.3 2223.46
  1340.1 2221.68  1347.7 2219.89  1376.1 2221.44  1404.9 2227.53  1464.1 2229.96
  1542.4 2244.56  1596.9  2246.9  1647.6 2254.14  1708.4 2260.12  1896.8 2274.28
  2247.5 2289.08  2437.3 2289.36  2608.2 2294.33  2740.1  2292.5  2817.5 2295.42
#Mann= 18 ,-1 , 0
       0     .04       0     470    .035       0     510     .04       0
     580    .035       0     690     .07       0    1150     .04       0
    1260    .035       0    1290     .04       0  1340.1    .045       0
  1376.1     .04       0    1380      .1       0    1690    .035       0
    1830      .1       0    1880    .035       0    2290      .1       0
    2520    .035       0    2630      .1       0    2660    .035       0
#XS Ineff= 2 , 0
          942.39 2232.61
Permanent Ineff=
       F       F
Bank Sta=1340.1,1376.1
XS Rating Curve= 0 ,0
Exp/Cntr(USF)=0,0
Exp/Cntr=0.3,0.1

Type RM Length L Ch R = 1 ,57747   ,460.7,443.4,401.2
XS GIS Cut Line= 3
     2132204.295      218310.776     2133332.768       219157.13
     2134014.517      220150.728
#Sta/Elev= 30
       0 2290.57    52.5  2291.7    88.6 2289.98   252.6 2269.18   314.9 2257.43
   380.5 2239.96   413.3 2234.79   439.6  2228.1   583.9 2224.06   731.5 2222.76
   879.2 2224.66   898.8 2223.58   915.2 2219.07   938.2 2222.73  1118.6  2223.8
  1128.5 2220.33  1164.6 2218.62  1174.4 2220.22  1190.8 2222.23  1207.2 2220.52
  1285.9 2222.32  1384.4 2230.76  1580.9 2264.09  1688.9 2277.46  1803.5 2284.72
  2062.2 2293.93  2252.1 2290.26  2383.1 2295.66  2494.4 2292.43  2615.6 2295.31
#Mann= 16 ,-1 , 0
       0     .04       0     170    .035       0     210      .1       0
     450    .035       0  1128.5    .045       0  1174.4    .035       0
    1190      .1       0 1460.59    .035       0 1580.59      .1       0
 1790.59    .035       0 1940.59      .1       0 1970.59    .035       0
 2060.59      .1       0 2320.59    .035       0 2420.59      .1       0
 2490.59    .035       0
#XS Ineff= 2 , 0
          627.81 2232.68
Permanent Ineff=
       F       F
Bank Sta=1128.5,1174.4
XS Rating Curve= 0 ,0
Exp/Cntr=0.3,0.1

Type RM Length L Ch R = 1 ,57304   ,478.4,476.9,468.2
XS GIS Cut Line= 3
2132424.64341683219477.5810814562133364.86013602219296.948312744
2133999.39063124220167.690890125
#Sta/Elev= 30
       0  2293.9      60 2301.22   100.1 2301.85   186.9 2292.54   213.6 2284.24
   240.4 2272.08   297.2 2241.49   307.2 2233.48   320.5 2232.72   333.9  2225.5
     354 2222.43   738.1 2222.83   768.2 2222.51   781.6 2217.95   795.3    2218
   826.1 2216.08   841.7 2218.18   859.7 2221.43   895.2 2218.84   908.5 2227.75
   955.3 2247.07  1054.2 2268.91  1137.7 2279.37  1238.3 2287.77  1465.8 2296.73
  1555.5 2296.32    1661  2286.7  1778.4  2296.7  1891.1 2291.15  2034.8 2296.39
#Mann= 12 ,-1 , 0
       0      .1       0     350    .035       0   795.3    .045       0
   841.7    .035       0     950      .1       0 1267.41    .035       0
 1327.41      .1       0 1437.41    .035       0 1447.41      .1       0
 1777.41    .035       0 1817.41      .1       0 1937.41    .035       0
Bank Sta=795.3,841.7
XS Rating Curve= 0 ,0
Exp/Cntr(USF)=0,0
Exp/Cntr=0.3,0.1

Type RM Length L Ch R = 1 ,56827   ,659.3,678.9,687.9
XS GIS Cut Line= 3
     2132498.892       219989.27     2133514.517      219624.686
      2133972.85      220171.561
#Sta/Elev= 30
       0    2345    88.6 2333.26   239.4 2304.23   285.4 2292.13     328 2276.31
   380.5  2260.9   475.6 2250.21   537.9 2246.47   564.1 2239.55   623.2 2217.62
   646.1  2220.2     656 2216.99   669.1 2214.68   695.3 2217.25     738 2221.06
   790.4 2218.12   842.9 2221.82   928.2 2220.74   941.3 2225.92  1000.4 2263.31
    1020 2272.31  1049.6 2282.92  1092.2 2290.52  1314.8 2295.36  1347.5 2292.58
  1399.8 2283.04  1429.3  2281.2  1543.9 2294.57  1648.6 2288.85  1792.6 2296.43
#Mann= 8 ,-1 , 0
       0     .04       0      20    .035       0     310      .1       0
     600     .07       0     656    .045       0   695.3     .07       0
     700      .1       0 1749.08    .035       0
Bank Sta=656,695.3
XS Rating Curve= 0 ,0
Exp/Cntr=0.3,0.1

Type RM Length L Ch R = 1 ,56148   ,507.5,511.1,489.7
XS GIS Cut Line= 2
     2132582.225       220176.77     2133971.763      220185.559
#Sta/Elev= 30
       0 2356.28    45.9 2346.16    98.3 2331.45   111.4 2326.11   127.8 2323.53
     213 2302.45   314.6 2261.84     354 2250.59   376.9 2245.82     485 2238.52
   550.6 2235.84   635.8 2227.59   770.2  2219.3   871.8  2217.6   884.9  2215.2
   894.7 2216.74     934 2215.17   966.8 2215.63   976.6 2217.46    1016 2217.05
  1035.6 2214.05  1058.6 2214.49  1068.4  2217.5  1133.9 2216.47  1140.5 2219.54
  1163.4 2235.82  1232.3 2280.21  1261.8 2294.39  1310.9  2297.9  1389.6 2297.51
#Mann= 5 ,-1 , 0
       0    .035       0      80      .1       0    1016    .045       0
  1068.4      .1       0    1360    .035       0
Bank Sta=1016,1068.4
XS Rating Curve= 0 ,0
Exp/Cntr=0.3,0.1

Type RM Length L Ch R = 1 ,55637   ,577.3,617.1,672.5
XS GIS Cut Line= 4
     2132604.576      220220.281     2133229.576      220263.684
 2133559.3877331220427.0610195582133938.23657963220376.733184017
#Sta/Elev= 30
       0 2353.71    36.5 2344.86    56.3 2336.76      76 2333.62   128.6 2316.26
   178.1 2304.16   289.8 2263.19   355.5 2243.92   382.8 2238.68   639.7 2225.59
   771.4 2222.23   811.8 2217.73   896.3  2220.3   932.6 2217.49   998.1 2220.41
  1011.4 2218.65  1018.8 2214.46  1027.6 2212.64  1044.5 2213.01  1051.1 2217.08
  1074.3 2218.76  1130.5 2218.71  1173.4 2214.51  1213.3 2214.87  1216.6 2216.57
  1236.4 2238.28  1256.3 2256.18  1286.1 2275.54  1345.6 2300.58  1376.7 2302.32
#Mann= 3 ,-1 , 0
       0      .1       0  1173.4    .045       0  1213.3      .1       0
Bank Sta=1173.4,1213.3
XS Rating Curve= 0 ,0
Exp/Cntr=0.3,0.1

Type RM Length L Ch R = 1 ,55020   ,552.8,520.4,491
XS GIS Cut Line= 3
     2132600.236      220268.024     2133164.472      220302.747
     2133229.576       220827.92
#Sta/Elev= 30
       0 2355.45    52.3 2342.04   114.4 2319.94   173.2 2303.45   215.7 2289.76
   235.3 2284.61   271.2 2272.61   310.4  2256.5   343.1 2248.71   369.2 2240.21
   388.8 2235.42     415 2231.61   437.9 2231.52   480.3 2228.77   555.5 2227.59
   627.4 2223.38     660 2222.43   689.4 2216.73   728.6 2217.34   784.2 2216.46
   790.7 2212.67   797.2 2212.02     843 2213.49   849.5 2216.93   859.3 2221.06
   878.9 2223.43     892 2226.79   921.4 2238.97   993.2 2264.58  1094.5 2296.48
#Mann= 3 ,-1 , 0
       0      .1       0   784.2    .045       0   849.5      .1       0
Bank Sta=784.2,849.5
XS Rating Curve= 0 ,0
Exp/Cntr=0.3,0.1

Type RM Length L Ch R = 1 ,54499   ,469.2,440.9,409.4
XS GIS Cut Line= 2
     2132487.388      220393.893     2133095.027      220884.344
#Sta/Elev= 30
       0 2370.98    26.1 2362.56    62.1 2346.19   107.8  2331.6   124.2 2323.17
   143.8 2310.18   166.6 2291.26   176.4 2284.82     183 2278.78   212.4 2261.01
   218.9 2254.43   225.4 2243.96   228.7 2239.99   258.1 2215.67   264.6 2212.49
   271.2 2211.21   297.3 2211.03   313.7 2212.93   320.2 2215.49   362.7 2218.51
   421.5 2219.58   480.3 2218.69   535.8 2224.13   578.3 2232.13   633.8  2239.2
   663.2 2244.48   699.2 2255.15   744.9 2270.55   764.5 2276.18   780.9 2279.11
#Mann= 3 ,-1 , 0
       0      .1       0   258.1    .045       0   320.2      .1       0
Bank Sta=258.1,320.2
XS Rating Curve= 0 ,0
Exp/Cntr=0.3,0.1
