HEC-RAS study SECONDCK.prj: SECONDCK

--- SECONDCK.g01 (geometry) --- (continued)

Type RM Length L Ch R = 1 ,54059   ,325,324.2,320.1
XS GIS Cut Line= 2
     2132396.243      220988.511     2133029.923       220984.17
#Sta/Elev= 30
       0 2347.79    58.8 2309.33    81.7 2291.98    88.2 2285.37    94.7 2277.43
   107.8 2265.42   117.6 2258.73   153.5 2230.99   173.1 2218.25   182.9 2213.16
   192.7 2209.78   225.4 2209.37   241.7 2210.08   254.8 2211.89   261.3 2213.72
   287.4 2217.63   323.4 2217.94   336.4 2219.56   346.2 2219.18   418.1 2221.84
     454 2223.86     503 2228.94   535.7 2236.06   545.5 2239.33   565.1 2243.99
   574.9 2247.56   591.2  2250.3   604.3 2256.03   623.9 2260.79   633.7 2264.14
#Mann= 3 ,-1 , 0
       0      .1       0   182.9    .045       0   261.3      .1       0
Bank Sta=182.9,261.3
XS Rating Curve= 0 ,0
Exp/Cntr=0.3,0.1

Type RM Length L Ch R = 1 ,53734   ,299.2,307.4,313
XS GIS Cut Line= 2
     2132413.604      221318.372      2132986.52       221287.99
#Sta/Elev= 30
       0 2321.15    16.4  2314.7    26.2 2309.79    85.2 2278.42   114.7 2260.22
     141 2242.81   173.8 2223.44   193.4 2214.22   209.8 2211.73   219.6 2209.02
   229.5 2207.97   255.7 2207.56   262.3 2207.62   272.1 2209.64   281.9 2210.38
   295.1  2213.4   301.6 2214.04     318 2213.06   327.8 2215.06   350.8 2216.47
     377  2219.2   386.8 2219.27   409.8 2222.49   429.5 2222.88   468.8 2227.31
     495 2233.59   514.7  2239.5   540.9 2248.31   563.9 2256.88   573.7 2261.29
#Mann= 3 ,-1 , 0
       0      .1       0   209.8    .045       0   281.9      .1       0
Bank Sta=209.8,281.9
XS Rating Curve= 0 ,0
Exp/Cntr=0.3,0.1

Type RM Length L Ch R = 1 ,53427   ,278.7,282.2,286.6
XS GIS Cut Line= 2
     2132413.604      221591.809     2132990.861      221622.191
#Sta/Elev= 30
       0 2282.98    19.6 2274.14    29.4 2268.94      62 2253.72    78.4 2248.69
   101.2 2240.83   107.8 2237.99   117.6  2235.3   153.5 2222.69   186.2 2215.74
   202.5  2215.6   218.8 2213.95   244.9 2212.94   264.5 2207.73   271.1 2207.38
   316.8 2207.72   329.8    2211   336.4 2211.48   339.6 2212.38   346.2 2214.33
   352.7 2215.19   372.3 2214.51   398.4  2215.6     405 2216.78   414.8 2219.67
   434.4 2227.64   460.5 2240.23   483.4  2250.4   545.4 2273.68   578.1 2288.14
#Mann= 5 ,-1 , 0
       0      .1       0   244.9    .045       0   339.6      .1       0
     450     .12       0     550      .1       0
Bank Sta=244.9,339.6
XS Rating Curve= 0 ,0
Exp/Cntr=0.3,0.1

Type RM Length L Ch R = 1 ,53145   ,247.3,256.1,263.6
XS GIS Cut Line= 2
     2132387.562      221813.163     2133016.902      221947.712
#Sta/Elev= 30
       0 2276.83    19.6 2268.22      49  2257.7    65.3 2249.62    75.1 2247.65
    84.9 2243.25   107.8 2235.52   114.3 2232.73   120.9 2228.66   133.9 2227.09
   166.6 2216.96     196 2212.83   225.4 2213.13   271.2 2215.66     281 2215.19
   307.1  2209.8   320.2 2211.38     330 2207.69   369.2 2207.51   375.7 2208.09
   382.2 2212.86   424.7 2240.53   460.6 2260.62     490 2276.23   516.2 2289.66
     539  2300.2   561.9 2309.15   591.3 2319.52     624  2333.6   643.6 2340.23
#Mann= 5 ,-1 , 0
       0      .1       0   320.2    .045       0   382.2      .1       0
     490     .12       0     590      .1       0
Bank Sta=320.2,382.2
XS Rating Curve= 0 ,0
Exp/Cntr=0.3,0.1

Type RM Length L Ch R = 1 ,52889   ,247.5,250,251.9
XS GIS Cut Line= 3
     2132328.418       221998.73     2132666.384      222133.916
      2133004.35      222269.101
#Sta/Elev= 30
       0 2303.36    29.5 2288.66    45.9 2279.22    55.8 2274.57    78.7 2262.72
    88.5 2257.04   108.2 2247.38     118 2243.44     141  2232.3   154.1  2228.3
     164 2224.47     200 2215.84   226.3  2212.9   259.1 2212.51     282 2213.97
   311.5    2214   334.5 2207.72   367.3 2207.68   380.4 2208.23   393.5 2211.88
   400.1  2214.7   419.8  2220.8   442.7 2229.15   485.3 2252.13   498.4 2260.21
   514.8 2268.56   550.9    2284   593.6 2300.62   682.1 2325.32     728 2333.11
#Mann= 5 ,-1 , 0
       0      .1       0   311.5    .045       0   400.1      .1       0
     674     .12       0     684      .1       0
Bank Sta=311.5,400.1
XS Rating Curve= 0 ,0
Exp/Cntr=0.3,0.1

Type RM Length L Ch R = 1 ,52639   ,469.5,473.6,478.4
XS GIS Cut Line= 3
     2132234.238      222213.547     2132566.177       222362.92
     2132898.116      222512.293
#Sta/Elev= 30
       0 2333.37    26.2 2318.23    75.4 2292.21   108.2 2271.77     118 2264.16
   131.2 2257.98     141 2251.02   170.5 2232.99   183.6 2229.44   196.8 2222.37
   213.2 2217.91   236.1  2215.2   259.1 2214.52   275.5 2211.74   318.1 2212.14
   347.6 2206.89   390.2 2207.11   393.5 2207.98   400.1 2212.16   409.9 2213.48
   426.3  2211.1   449.3 2213.65   478.8  2225.8   524.7 2248.77   567.3  2265.8
   613.2 2278.96     646 2289.75   701.8 2304.13   718.2 2309.67     728 2310.54
#Mann= 5 ,-1 , 0
       0      .1       0   318.1    .045       0   400.1      .1       0
     474     .12       0     694      .1       0
Bank Sta=318.1,400.1
XS Rating Curve= 0 ,0
Exp/Cntr=0.3,0.1

Type RM Length L Ch R = 1 ,52165   ,233.2,272,311.5
XS GIS Cut Line= 3
     2132124.284      222432.122     2132187.909       222694.24
     2132685.759      222963.369
#Sta/Elev= 30
       0 2298.15    35.8 2294.15   113.7 2279.64   149.5 2275.19   172.2 2269.52
   204.7 2260.31     221 2254.49   269.7  2231.3   282.8 2223.84   299.2 2216.45
     309 2213.41     345 2210.64   390.8    2214   403.8 2213.42   420.2 2214.65
     430 2214.21   443.1 2211.89   462.7 2208.39   498.7 2206.04   524.9 2208.93
     538 2212.63   655.7  2253.6   717.9  2272.6   740.8 2281.52   750.6 2286.45
   763.7 2289.39   773.5  2295.6   796.4 2306.56   806.2 2308.84   835.7 2323.54
#Mann= 3 ,-1 , 0
       0      .1       0   443.1    .045       0     538      .1       0
Bank Sta=443.1,538
XS Rating Curve= 0 ,0
Exp/Cntr=0.3,0.1

Type RM Length L Ch R = 1 ,51893   ,236.8,265.5,292.8
XS GIS Cut Line= 2
     2132076.946      222468.767     2132287.736      223306.219
#Sta/Elev= 30
       0 2286.28    26.2 2282.72    68.7 2274.62   114.5 2270.25   222.4 2255.97
   232.2 2253.73   251.9 2247.35   310.8 2217.98   323.8 2213.22   333.6 2210.88
   343.5 2210.02   359.8 2210.37   444.9 2214.42     458  2213.5   467.8 2213.93
   484.1  2212.4   500.5 2213.15   513.6 2209.94   529.9 2206.04   536.5 2205.88
   569.2 2206.28   575.7 2207.44   582.3 2210.54   598.6 2218.63   624.8 2226.93
   693.5 2264.82   722.9 2278.62   762.2 2294.84   804.7 2315.06   863.6 2340.58
#Mann= 3 ,-1 , 0
       0      .1       0   513.6    .045       0   582.3      .1       0
Bank Sta=513.6,582.3
XS Rating Curve= 0 ,0
Exp/Cntr=0.3,0.1

Type RM Length L Ch R = 1 ,51628   ,469.2,495.2,520.4
XS GIS Cut Line= 3
     2132015.345      222474.651     2132022.979      222824.448
     2131875.409      223258.476
#Sta/Elev= 30
       0 2273.41    26.2 2267.54    52.3 2262.57   137.3  2252.3   196.2 2243.92
   300.8 2236.47     327 2232.84   343.3 2228.26   372.8 2215.06   389.2 2210.62
   461.2 2209.33     471  2210.1   484.1  2212.5   500.5 2213.28   513.6 2211.88
   520.2 2208.91   539.8 2204.92   549.6 2204.53   569.3 2204.77   592.2 2206.15
   598.7 2207.55     602 2209.24   608.6 2213.94   624.9  2230.1     661 2261.02
   703.5 2294.19   719.9 2305.56   746.1  2320.9   788.7    2349   808.3 2361.02
#Mann= 4 ,-1 , 0
       0      .1       0   520.2    .045       0     602      .1       0
  789.88     .04       0
Bank Sta=520.2,602
XS Rating Curve= 0 ,0
Exp/Cntr=0.3,0.1

Type RM Length L Ch R = 1 ,51132   ,346,354.7,362
XS GIS Cut Line= 3
     2131892.385       222418.94     2131601.972      222685.559
     2131489.125      222776.705
#Sta/Elev= 30
       0 2251.36    29.3  2243.6    81.4 2226.78    94.5 2223.06   117.3 2218.18
   146.6 2213.47   169.4 2210.51   205.3 2208.56   211.8 2208.68   221.6 2207.79
   244.4 2208.36   260.6 2206.56   286.7 2207.72   296.5 2207.21   309.5 2204.36
     316 2203.56   345.4 2203.47   361.7 2203.51   364.9    2204   368.2 2205.35
   371.4  2207.5   400.7 2232.22   432.9 2256.15     491 2293.42   497.4  2298.5
   500.6 2300.36     520 2309.78   532.8 2317.02   536.1 2318.22   539.3 2317.97
#Mann= 3 ,-1 , 0
       0      .1       0   296.5    .045       0   371.4      .1       0
Bank Sta=296.5,371.4
XS Rating Curve= 0 ,0
Exp/Cntr=0.3,0.1

Type RM Length L Ch R = 1 ,50778   ,292.2,303.4,311.9
XS GIS Cut Line= 2
      2131755.76      222154.429     2131306.833      222442.504
#Sta/Elev= 30
       0 2261.38    26.2 2249.21    45.8 2239.53    68.7 2229.62   104.7 2216.25
   114.5 2213.04   130.9  2209.1   150.5 2206.36   160.4 2205.99     180 2207.38
   255.2 2208.71   278.2 2205.41   294.5 2205.11   301.1 2203.88   310.9 2201.87
   317.4  2201.4   356.7 2202.38   379.6 2201.52   386.2 2201.86     396 2203.75
   405.8 2204.25   418.9 2207.62     432 2212.82   441.8 2217.54   490.9 2250.11
     504 2259.41   513.8 2268.14     517 2270.36   523.6 2274.64   533.4 2280.12
#Mann= 6 ,-1 , 0
       0     .12       0     100      .1       0     180     .12       0
     220      .1       0   301.1    .045       0     396      .1       0
Bank Sta=301.1,396
XS Rating Curve= 0 ,0
Exp/Cntr=0.3,0.1

Type RM Length L Ch R = 1 ,50474   ,314.3,320.2,321.7
XS GIS Cut Line= 3
     2131652.018      221934.918     2131317.017      222077.294
     2131089.819      222169.066
#Sta/Elev= 30
       0 2262.07    13.1 2257.38    49.2 2240.03   111.5 2215.68   124.6 2212.95
   160.7 2209.57   186.9 2208.48   209.9 2205.98   255.8 2206.32   275.5 2203.68
   298.4 2205.27   308.2 2205.23   321.4 2203.42   331.2 2201.12   380.3 2200.38
   396.7 2206.05   399.9 2207.24   406.5 2207.97   426.1 2206.88   448.9    2207
   455.5 2208.19   465.3 2212.22   475.1 2217.69   514.3 2244.92   524.1 2263.17
   530.6 2269.35     547 2281.12   573.1 2297.18   592.7 2304.87     609 2309.32
#Mann= 5 ,-1 , 0
       0      .1       0      80     .12       0     190      .1       0
   308.2    .045       0   396.7      .1       0
Bank Sta=308.2,396.7
XS Rating Curve= 0 ,0
Exp/Cntr=0.3,0.1

Type RM Length L Ch R = 1 ,50154   ,494.3,496,493.4
XS GIS Cut Line= 3
     2131545.548      221656.913      2131415.34      221713.337
     2130873.938      221890.083
#Sta/Elev= 30
       0 2289.33    61.3 2255.29    87.1 2238.54   125.8 2220.76   138.7 2216.21
   174.6 2208.72   256.5 2205.19   269.6 2202.42   292.5 2202.85   302.3 2199.29
   308.8 2199.22   354.7 2199.56   364.5 2203.66   397.2 2203.18   433.2 2205.91
     466 2205.36   475.8 2207.22   492.1 2215.85     502 2224.33   511.8 2227.71
   518.3 2233.85     538 2256.33     551 2267.67   577.2 2284.37   593.6 2293.16
   603.4 2297.06   623.1 2301.34   639.4 2302.27   675.4 2301.75   711.4 2299.35
#Mann= 6 ,-1 , 0
       0     .12       0      10      .1       0      80     .12       0
  181.91      .1       0   292.5    .045       0   364.5      .1       0
Bank Sta=292.5,364.5
XS Rating Curve= 0 ,0
Exp/Cntr=0.3,0.1

Type RM Length L Ch R = 1 ,49658   ,407.1,379.2,314.1
XS GIS Cut Line= 3
     2131337.215      221244.587     2130933.569      221405.177
     2130763.215      221749.845
#Sta/Elev= 30
       0 2261.64    26.1 2251.23    39.2 2247.72    58.8  2243.6    75.1    2238
    94.7 2228.98   143.7 2209.12   166.6 2204.52   199.2 2201.21   218.8 2202.79
   254.8 2203.48   287.4    2203   300.5 2204.74   320.1 2203.54   349.5 2198.84
   369.1 2199.94   401.8 2203.78   411.6 2207.79   427.9 2218.66   434.4 2223.87
   470.3 2242.92   483.3 2250.37   499.6  2261.1   519.1 2268.06   541.9 2273.55
   564.8  2275.7   610.4 2278.48   646.2 2279.16   779.8 2275.51   818.9 2273.82
#Mann= 4 ,-1 , 0
       0      .1       0     270     .12       0   320.1    .045       0
   401.8      .1       0
Bank Sta=320.1,401.8
XS Rating Curve= 0 ,0
Exp/Cntr=0.3,0.1

Type RM Length L Ch R = 1 ,49279   ,382.1,360.4,329.5
XS GIS Cut Line= 2
     2130937.909       220819.24     2130736.802      221707.039
#Sta/Elev= 30
       0 2297.81    22.9  2287.1    39.3 2280.84    75.3 2263.72    85.1 2260.22
   137.5  2235.3   170.3  2217.1   183.4 2208.84   189.9 2203.21   199.7 2197.05
   216.1 2196.45   229.2 2196.71     262 2202.25   278.3 2200.61   294.7 2201.08
   311.1 2203.09   324.2 2202.29   343.8 2203.79   363.5  2199.8   376.6 2200.82
   392.9 2204.17   445.3 2202.23   455.2 2206.11   494.4 2229.58   504.3 2234.56
   563.2 2252.44   586.1 2255.39   717.1 2264.75   766.2 2266.89   910.3 2266.57
#Mann= 5 ,-1 , 0
       0      .1       0      60     .12       0     160      .1       0
   189.9    .045       0     262      .1       0
Bank Sta=189.9,262
XS Rating Curve= 0 ,0
Exp/Cntr=0.3,0.1

Type RM Length L Ch R = 1 ,48918   ,336.3,318.1,291.2
XS GIS Cut Line= 3
     2130451.798      220888.684      2130642.77      221305.351
     2130639.744      221706.596
#Sta/Elev= 30
       0 2316.12    29.5 2301.44    42.6 2296.66   101.5 2271.24   121.1 2261.43
   134.2 2256.45   147.3  2249.6   180.1 2228.73     203 2217.16   219.4  2211.1
     239 2199.62   245.5  2195.8   248.8 2194.96   271.7 2194.35   284.8 2194.69
   307.8 2199.63   320.8 2200.99   340.5 2200.84   353.6 2201.88   392.9 2201.78
   438.7 2205.03   461.6  2208.9   477.9 2212.71   510.5 2224.52   530.1 2228.89
   562.7 2233.94   634.5 2241.41     690 2245.58   758.5 2247.83   859.6 2249.57
#Mann= 5 ,-1 , 0
       0      .1       0     110     .12       0     239    .045       0
   307.8     .12       0     310      .1       0
Bank Sta=239,307.8
XS Rating Curve= 0 ,0
Exp/Cntr=0.3,0.1

Type RM Length L Ch R = 1 ,48600   ,321,311.3,297.7
XS GIS Cut Line= 3
     2130085.305      221136.847     2130499.541      221457.261
     2130595.117      221740.687
#Sta/Elev= 30
       0 2330.75    13.1  2328.7    65.5 2313.84    75.3 2310.38    88.4 2304.43
   101.5 2296.91   104.7 2294.14   111.3 2285.54   114.6 2282.42     144 2266.06
   196.4 2245.65     216 2236.07   242.2 2224.99   255.3 2218.16   297.8 2203.22
   304.4  2199.1   310.9 2195.86   320.8 2194.24   350.2 2193.81   376.4 2194.22
   402.6 2198.94   412.4 2199.54     432 2199.16   481.1 2200.97   500.8 2205.28
     527 2214.68   556.2 2220.02   660.2  2229.7   731.8 2234.38   822.8 2242.93
#Mann= 7 ,-1 , 0
       0    .035       0      30      .1       0      50    .035       0
     150      .1       0   304.4    .045       0   402.6     .12       0
     520      .1       0
Bank Sta=304.4,402.6
XS Rating Curve= 0 ,0
Exp/Cntr=0.3,0.1

Type RM Length L Ch R = 1 ,48289   ,318.7,309.6,296.3
XS GIS Cut Line= 2
     2129913.604      221474.622     2130554.057      221791.886
#Sta/Elev= 30
       0 2303.25    55.7 2299.35   147.5 2295.19   173.8 2296.29   193.4 2293.56
     200 2290.85   203.3 2287.96   206.6 2282.08   216.4 2257.43   219.7 2252.39
   226.2 2246.98   232.8 2238.22   239.3  2232.5     282 2204.98   304.9 2198.89
   308.2 2197.16   314.7 2193.36   321.3 2192.02   354.1 2191.67   380.3 2194.31
   393.4 2197.71   403.3 2198.56   432.8 2198.38   452.4 2196.31   468.8  2197.8
   504.9 2197.61     541 2204.82     600 2219.21   678.7 2229.41   714.7  2235.8
#Mann= 4 ,-1 , 0
       0      .1       0   308.2    .045       0   393.4     .12       0
     440      .1       0
Bank Sta=308.2,393.4
XS Rating Curve= 0 ,0
Exp/Cntr=0.3,0.1

Type RM Length L Ch R = 1 ,47979   ,396.9,386.1,373.8
XS GIS Cut Line= 3
     2129785.128      221844.026     2130140.621      221923.387
     2130495.029      222006.023
#Sta/Elev= 30
       0 2262.78      26 2260.43    58.5 2261.07   130.1  2273.4   152.8 2276.36
   208.1 2279.53   227.6 2277.24   243.9  2271.4   266.7 2258.56   269.9  2255.6
   282.9  2236.8   286.2 2233.14   312.2  2213.9   328.5 2195.52     335 2190.52
   341.5 2189.12   367.5 2189.26   387.2 2195.07   410.1 2197.03   439.6 2195.05
   475.7 2196.48   505.2 2196.09   534.7 2194.26   551.1    2195   564.2 2196.85
   580.6 2200.74   636.4 2216.57   659.3 2220.73   695.4 2225.43   728.2 2231.94
#Mann= 5 ,-1 , 0
       0     .04       0      30      .1       0   328.5    .045       0
   387.2     .12       0  504.24      .1       0
Bank Sta=328.5,387.2
XS Rating Curve= 0 ,0
Exp/Cntr=0.3,0.1

Type RM Length L Ch R = 1 ,47593   ,479,449.4,400.6
XS GIS Cut Line= 2
     2129748.673      222312.295      2130454.78      222284.547
#Sta/Elev= 30
       0 2237.96    91.6 2258.24     121 2259.62   130.9  2261.4   147.2  2260.5
   150.5 2259.33   173.4 2245.47   202.8 2223.32     229 2209.25   248.6 2201.26
   268.3 2198.62   278.1 2194.74   291.2 2188.88   297.7 2188.33   317.3  2188.7
   346.8 2194.07   376.2 2195.55   428.6 2192.82   471.1 2192.24   487.5 2193.38
   516.9 2191.97   536.5  2193.6   556.2 2192.62   572.5 2192.97   588.9 2197.96
   608.5 2210.44   618.3 2214.31   628.1 2216.51   690.3 2224.48   706.6 2228.14
#Mann= 7 ,-1 , 0
       0     .04       0      60    .035       0     160      .1       0
   278.1    .045       0   346.8      .1       0     360     .12       0
     460      .1       0
Bank Sta=278.1,346.8
XS Rating Curve= 0 ,0
Exp/Cntr=0.3,0.1

Type RM Length L Ch R = 1 ,47144   ,559.6,552.5,520.6
XS GIS Cut Line= 3
     2129817.764      222771.954     2130208.743      222711.601
     2130438.777       222386.08
#Sta/Elev= 30
       0  2254.8   143.9 2270.56     170 2275.11   192.9 2277.67   209.2 2278.25
   245.2 2272.86   258.3 2272.47   264.8 2270.98   281.2 2261.73   304.1  2253.1
   320.4 2243.61   349.8 2229.18   382.5 2217.27   392.3 2212.72   408.7 2202.55
   421.8 2192.01     425 2190.77   438.1 2186.02   444.6 2185.73   454.4 2186.04
   467.5 2188.74   487.1 2190.81   526.3  2187.4   555.7 2188.28   575.3 2192.26
   588.4 2196.97   601.4 2199.62   624.3 2201.22   748.5 2221.56   794.2 2226.56
#Mann= 6 ,-1 , 0
       0      .1       0     210    .035       0     290      .1       0
     425    .045       0   487.1     .12       0  605.61      .1       0
Bank Sta=425,487.1
XS Rating Curve= 0 ,0
Exp/Cntr=0.3,0.1

Type RM Length L Ch R = 1 ,46591   ,446.8,471.6,508.2
XS GIS Cut Line= 3
     2130167.944      222954.656     2130677.493      222945.976
     2130768.638      222533.649
#Sta/Elev= 30
       0 2236.64    91.5 2237.32   143.7 2238.75   209.1 2238.03   254.8 2233.07
     330 2234.09   336.5 2232.64   346.3  2227.2   349.6 2226.35   382.2 2226.75
   405.1 2224.97   431.2 2227.23   457.4 2232.85   463.9 2233.44     526 2234.89
   545.6 2234.14   578.4 2222.79   624.2 2204.49   630.7  2200.4   647.1 2184.36
   650.4 2182.29   696.2 2182.06   712.6 2181.28     729 2182.36   748.6 2185.92
   784.6 2187.38   840.2 2194.43   853.3 2198.12   902.4 2218.68   931.9 2227.66
#Mann= 7 ,-1 , 0
       0      .1       0     330     .06       0  519.62      .1       0
  589.62    .035       0  619.62      .1       0   696.2    .045       0
     729      .1       0
Bank Sta=696.2,729
XS Rating Curve= 0 ,0
Exp/Cntr=0.3,0.1

Type RM Length L Ch R = 1 ,46120   ,296.1,316.8,341.1
XS GIS Cut Line= 3
     2130180.965      222972.886     2130816.381       223015.42
     2131327.017      222687.186
#Sta/Elev= 30
       0 2231.72     160  2229.1   182.9 2227.32     209 2223.24   290.7 2216.32
     320 2218.77   385.4 2221.46   476.8 2230.41   512.7  2230.1   571.5 2221.24
   653.2  2199.6   666.2 2193.27   679.3 2184.73   692.3 2181.88   845.7 2184.98
   878.4  2183.5   914.2 2184.09   950.1 2181.13     973 2183.04  1021.9 2180.79
  1041.5 2181.98  1067.6 2178.88  1087.2  2179.1    1097    2183  1116.6 2204.77
  1119.8 2206.79  1132.9 2208.25  1142.7 2213.76  1172.1 2225.06  1243.9  2261.1
#Mann= 7 ,-1 , 0
       0      .1       0     320     .06       0     520      .1       0
     620    .035       0  726.84      .1       0  1041.5    .045       0
    1097      .1       0
Bank Sta=1041.5,1097
XS Rating Curve= 0 ,0
Exp/Cntr=0.3,0.1

Type RM Length L Ch R = 1 ,45803   ,406.5,443.1,495.4
XS GIS Cut Line= 2
     2130201.798      222993.719      2131415.34      223097.886
#Sta/Elev= 30
       0 2226.33   124.4 2223.15   144.1 2221.52   183.4 2213.83   229.2 2209.84
   265.2 2212.54   343.8 2211.67   448.6 2220.95   484.6 2220.99   510.8  2219.4
   543.5 2214.65   592.6 2204.34     609 2199.54   635.2 2198.13   638.5 2197.13
   658.1 2184.52   667.9 2182.45   694.1 2181.04   713.8 2182.86     740 2180.97
   877.5 2183.36   926.6 2181.76     943 2178.23   952.8  2177.7   988.8 2177.96
  1011.7 2181.65  1044.5 2184.88    1087 2200.31  1159.1 2231.42    1218  2263.1
#Mann= 8 ,-1 , 0
       0      .1       0     300     .06       0     500     .04       0
     600      .1       0     700    .035       0     890      .1       0
   926.6    .045       0  1011.7      .1       0
Bank Sta=926.6,1011.7
XS Rating Curve= 0 ,0
Exp/Cntr=0.3,0.1

Type RM Length L Ch R = 1 ,45360   ,325.9,353.7,380.4
XS GIS Cut Line= 3
     2130188.777      223011.948     2130725.236      223071.844
     2131024.715      223627.399
#Sta/Elev= 30
       0 2221.66    52.3  2221.1    98.1 2218.26   143.9 2213.63   173.4 2208.28
   206.1 2204.26   238.8 2207.18   268.3 2205.05     350  2203.5   451.5 2209.64
   516.9  2209.7   539.8 2207.88     566 2201.01   595.4 2195.51   631.4 2191.25
   644.4 2184.87   654.2 2182.17   703.3 2179.31   765.4 2178.11   788.3 2174.89
   843.9 2177.58   925.7    2178   941.3 2176.09   974.7 2176.49   981.3 2177.87
   987.8 2182.84   997.6 2193.82  1000.9 2195.85  1043.4 2211.87  1170.9 2270.58
#Mann= 9 ,-1 , 0
       0      .1       0     220     .06       0     310     .04       0
     410     .06       0     510     .04       0  679.79     .06       0
  729.79      .1       0   925.7    .045       0   981.3      .1       0
Bank Sta=925.7,981.3
XS Rating Curve= 0 ,0
Exp/Cntr=0.3,0.1

Type RM Length L Ch R = 1 ,45006   ,506.3,496.4,488
XS GIS Cut Line= 4
     2130162.736      223019.7612130664.08745597223108.436583994
2130576.23300171223478.6795549122130608.77779998223738.998071994
#Sta/Elev= 30
       0  2219.3    67.9 2218.18   101.6 2213.82   124.3 2213.28   197.8  2200.1
   227.8  2201.3   254.5 2195.57   291.1 2195.27   314.4 2200.02   377.7 2201.78
   509.1 2200.35   615.3 2187.69   638.9 2187.67   655.8 2184.62   682.7 2175.58
   692.9 2173.87   786.9 2173.58   800.8 2171.25   827.8 2171.34   837.9 2173.54
   851.3 2178.58   861.5  2180.2   871.6 2185.91     885 2195.84   941.4 2230.97
   960.1 2248.26  1073.6  2314.1  1107.1 2321.52  1127.7 2319.23    1152 2312.29
#Mann= 8 ,-1 , 0
       0      .1       0     100     .06       0     340     .04       0
     440     .06       0  539.13     .04       0  639.13      .1       0
   786.9    .045       0   837.9      .1       0
Bank Sta=786.9,837.9
XS Rating Curve= 0 ,0
Exp/Cntr=0.3,0.1

Type RM Length L Ch R = 1 ,44510   ,387.6,371.3,354.7
XS GIS Cut Line= 3
     2130126.277      223022.365     2130139.298      223616.115
     2130334.611      223741.115
#Sta/Elev= 30
       0 2217.24    39.2 2204.74    51.6 2203.17      68 2197.65    87.7 2196.36
   117.2 2191.06   143.5 2190.54   163.2 2188.13   182.9 2182.59   212.12171.385
   225.5 2167.88   232.1 2167.69   258.3  2167.7   267.6 2171.24   281.3 2175.04
   284.6 2174.87   294.4 2170.66   304.3 2169.84   330.5 2170.57     370 2168.73
   412.6 2171.44   504.8 2169.49   550.4 2171.76   572.3 2174.37   593.9 2174.45
     623 2181.84   677.6 2190.45   724.5 2202.36   759.5 2214.46   825.8 2241.64
#Mann= 7 ,-1 , 0
       0      .1       0      20     .06       0   212.1    .045       0
   267.6      .1       0     410     .06       0     510    .035       0
  613.89      .1       0
Bank Sta=212.1,267.6
XS Rating Curve= 0 ,0
Exp/Cntr=0.3,0.1

Type RM Length L Ch R = 1 ,44139   ,205.7,202.3,197.4
XS GIS Cut Line= 3
     2129760.826      223052.747     2129750.409      223257.608
     2130069.854      223896.497
#Sta/Elev= 30
       0 2223.81    39.1 2220.32    65.1 2216.41    97.7 2214.48     127 2208.73
   159.5 2200.42   198.6 2192.94   224.8 2190.78   241.2 2184.51   257.6 2168.37
   264.1 2165.74   275.9 2165.14   296.9 2165.29   313.2 2169.27   323.1  2168.5
   388.6 2169.96   408.3 2166.88   427.9 2167.93   450.9 2166.88   470.5 2168.19
   486.9 2166.69   545.9 2168.75   640.9 2169.17     677 2166.96   699.9 2168.71
   739.2 2168.19   794.9 2173.35   814.6 2179.09   847.3 2183.81   919.4 2188.13
#Mann= 8 ,-1 , 0
       0      .1       0   257.6    .045       0   313.2      .1       0
  405.13    .035       0  625.13      .1       0  735.13     .04       0
  775.13      .1       0  845.13     .06       0
Bank Sta=257.6,313.2
XS Rating Curve= 0 ,0
Exp/Cntr=0.5,0.3

Type RM Length L Ch R = 1 ,43936   ,74.4,73.4,73
XS GIS Cut Line= 3
2129694.61301816 223017.501639192129518.82236989223285.797803702
     2129970.027       223975.49
#Sta/Elev= 30
       0 2220.49    53.5  2217.4    83.2 2213.08    90.4 2210.73   104.6 2203.18
   161.3 2196.21   196.4 2185.22   245.1 2173.58   322.4 2170.67   406.2 2172.24
   428.3 2169.96   465.7 2170.55   483.2 2169.22     491 2166.36   498.4  2163.5
   505.8 2163.36   541.3 2163.44   550.8 2166.52   558.3 2168.23   581.6 2168.51
   676.4 2165.79   694.9 2167.54   726.2 2167.77   749.9 2167.77   769.4 2165.97
   894.8 2166.76   941.9 2174.81   969.3 2177.36   996.8 2174.88  1144.9 2183.62
#Mann= 9 ,-1 , 0
       0     .06       0      30      .1       0  380.76     .08       0
  490.76     .06       0     491    .045       0   550.8     .08       0
  610.76     .06       0 1030.76     .04       0 1080.76     .06       0
#XS Ineff= 4 ,-1
       0     310    2167     310     460    2172     580     730    2172
     730  1144.9    2167
Permanent Ineff=
       F       F       F       F
Bank Sta=491,550.8
XS Rating Curve= 0 ,0
Exp/Cntr=0.5,0.3

Type RM Length L Ch R = 1 ,43863   ,274.1,263.1,247.4
XS GIS Cut Line= 3
2129090.64995005223194.651246594     2129472.631       223350.49
     2129912.736      224014.552
#Sta/Elev= 30
       0 2218.12    39.5 2212.55   113.9 2198.51   170.6 2181.49   188.3 2180.31
   220.2 2175.56   330.1 2167.87     408 2167.67   452.5 2164.87   470.3 2168.02
   511.9 2167.02   520.1 2170.74   541.3 2171.49   559.4 2169.59   567.4 2166.78
   574.5  2164.1   588.7 2163.35   606.9  2163.6   618.8  2166.7   623.9  2169.5
   627.9 2169.93   647.9 2167.52   701.9 2168.13   750.8 2166.28   887.7 2164.45
   978.2 2165.68  1068.7 2168.59  1105.7 2174.37  1141.4 2174.75  1209.2 2180.81
#Mann= 14 ,-1 , 0
       0      .1       0      30    .035       0     110      .1       0
     140    .035       0     350     .06       0  492.55     .08       0
   567.4    .045       0   618.8     .08       0  632.55      .1       0
  662.55     .06       0  752.55    .035       0  842.55     .06       0
  982.55    .035       0 1022.55     .06       0
#XS Ineff= 4 ,-1
       0     400    2167     400   566.7    2172   623.3     775    2172
     775  1209.2    2167
Permanent Ineff=
       F       F       F       F
Bank Sta=567.4,618.8
XS Rating Curve= 0 ,0
Exp/Cntr=0.5,0.3

Type RM Length L Ch R = 1 ,43600   ,670.3,647.5,604.9
XS GIS Cut Line= 3
     2128764.298      223563.163      2129267.77      223597.886
     2129899.715      224056.219
#Sta/Elev= 30
       0 2224.34    49.2 2221.15   206.5 2219.06   278.6 2213.27   298.2 2210.45
   337.5 2199.88   360.5 2196.13   403.1 2190.56   475.2  2185.7   521.1 2181.38
   550.6 2176.34   576.8 2168.51   586.7 2166.62     626 2164.78   642.4 2161.52
     672 2161.95   685.1 2164.65   691.6 2167.35   714.6 2164.73   868.8  2165.1
   996.7 2162.56  1026.2 2165.47  1045.9 2164.33  1111.5 2163.93  1190.2 2166.35
  1206.6 2168.75  1216.4 2172.54  1226.3 2174.46    1246 2174.92  1285.3 2178.51
#Mann= 9 ,-1 , 0
       0     .06       0     160    .035       0  564.67     .06       0
     626    .045       0   685.1      .1       0  724.67     .06       0
  814.67    .035       0 1174.67     .06       0 1224.67     .04       0
Bank Sta=626,685.1
XS Rating Curve= 0 ,0
Exp/Cntr=0.3,0.1

Type RM Length L Ch R = 1 ,42952   ,383.1,386.1,387.4
XS GIS Cut Line= 2
     2128979.576      224396.497     2129920.548       224167.33
#Sta/Elev= 30
       0 2203.73      36    2200      72 2194.86   114.5 2193.36   153.8 2188.93
   212.7 2185.74   320.6 2176.93   353.4 2174.97   369.7 2172.17   386.1 2165.93
   399.2 2162.91   438.4 2161.26   451.5  2159.5   464.6 2158.06   513.7 2157.33
     530 2158.87   562.8 2160.88   575.8 2160.81   624.9 2158.38   641.3 2156.81
   670.7 2159.21   687.1 2162.09   749.3 2162.29   791.8 2161.47   870.3 2162.81
   880.1  2165.7   899.8 2175.59   916.1 2176.37   929.2 2179.65   968.5 2183.59
#Mann= 9 ,-1 , 0
       0     .12       0      50      .1       0     250     .12       0
   451.5    .045       0     530     .12       0     550      .1       0
     650     .12       0     760      .1       0     960     .06       0
Bank Sta=451.5,530
XS Rating Curve= 0 ,0
Exp/Cntr=0.3,0.1

Type RM Length L Ch R = 1 ,42566   ,371.6,377,402.8
XS GIS Cut Line= 2
     2129177.493      224712.469      2129955.27      224580.524
#Sta/Elev= 30
       0 2252.99    22.9 2252.74    49.1 2247.64    81.8 2233.42   111.3  2216.5
   130.9 2206.88   160.4 2195.26   209.5 2180.24   255.3  2172.5   294.6 2156.97
   304.4 2155.16   350.2 2154.52   373.2 2155.79   392.8  2157.5   409.2 2154.44
   438.6 2155.62   471.4 2154.29   507.4 2157.91   572.8 2157.78   595.8 2155.97
   638.3 2157.35   644.9 2158.62   654.7 2163.11   684.1 2179.83   703.8 2186.24
   710.3 2187.42   733.2 2187.92   749.6 2193.08   759.4 2194.67   788.9 2196.76
#Mann= 5 ,-1 , 0
       0     .12       0   294.6    .045       0   373.2      .1       0
     640     .04       0     740      .1       0
Bank Sta=294.6,373.2
XS Rating Curve= 0 ,0
Exp/Cntr=0.3,0.1

Type RM Length L Ch R = 1 ,42189   ,354.2,384.2,404.6
XS GIS Cut Line= 3
     2129226.865      224864.595     2129476.104      225000.663
      2129955.27      225070.108
#Sta/Elev= 30
       0 2211.22    29.4 2200.46    68.5  2183.1    78.3 2180.22    94.6  2177.3
   169.7 2170.41   182.8 2168.32   199.1 2167.83   241.5 2163.62   277.4 2157.17
   329.8 2154.69   349.4 2154.84   362.5  2152.2   375.6 2153.29   395.2 2151.29
   401.7 2150.08   418.1 2149.87   467.2 2150.31     477 2151.36   499.9 2154.28
   529.3 2153.68     549 2157.77   581.7 2160.48   647.1 2169.96   656.9 2172.83
   673.3 2179.59   692.9 2190.18   699.4 2192.26   728.9 2194.13   768.1 2194.39
#Mann= 6 ,-1 , 0
       0     .12       0     220      .1       0  323.96     .12       0
   395.2    .045       0     477      .1       0  723.96     .06       0
Bank Sta=395.2,477
XS Rating Curve= 0 ,0
Exp/Cntr=0.3,0.1

Type RM Length L Ch R = 1 ,41805   ,416.2,442.9,452.8
XS GIS Cut Line= 2
     2129179.884      225088.699     2129715.687      225559.691
#Sta/Elev= 30
       0 2175.24    39.3 2171.42   104.7 2163.28   117.8  2160.5     144 2153.38
   153.8 2151.63     180 2152.09   193.1 2152.55   212.7 2151.47   229.1 2152.56
     252  2151.4   278.2  2151.4   294.5    2149   314.2 2149.06   346.9 2152.62
   369.8 2152.74   386.1 2150.65   412.3 2149.59   422.1 2147.25   428.7 2146.65
     432 2146.84   448.3 2150.85   471.2 2164.58   510.5 2183.93   523.6 2191.98
   530.1 2194.07   566.1 2194.27   605.4 2198.19   644.7 2201.05   713.4 2207.92
#Mann= 7 ,-1 , 0
       0     .12       0      30      .1       0     180     .12       0
   386.1    .045       0   448.3     .12       0     470      .1       0
     710     .04       0
Bank Sta=386.1,448.3
XS Rating Curve= 0 ,0
Exp/Cntr=0.3,0.1

Type RM Length L Ch R = 1 ,41362   ,478.6,467.5,450
XS GIS Cut Line= 2
     2128962.215      225208.997     2129268.873       225893.77
#Sta/Elev= 30
       0    2180   101.6 2161.63   134.3  2149.1   140.9  2147.9   163.8 2147.52
   183.5  2149.5   222.8 2150.38   275.2  2149.1   317.8 2149.71   327.6  2149.4
   340.8 2146.46   350.6 2146.32   360.4 2143.88   370.2 2143.51   399.7 2146.15
   435.8  2143.6   448.9 2144.06   458.7 2146.19   478.4 2148.57   501.3 2148.79
   511.1 2150.74   530.8 2159.34   543.9 2161.59   563.6 2177.07   576.6 2183.59
   632.4 2185.93   681.5 2178.52   704.4 2179.11   724.1 2183.18   750.3 2183.02
#Mann= 4 ,-1 , 0
       0      .1       0   399.7    .045       0   458.7     .12       0
     540      .1       0
Bank Sta=399.7,458.7
XS Rating Curve= 0 ,0
Exp/Cntr=0.3,0.1

Type RM Length L Ch R = 1 ,40894   ,520.5,497.7,463.7
XS GIS Cut Line= 2
     2128451.798      225514.552     2129059.353      226036.603
#Sta/Elev= 30
       0 2252.54      36 2237.45    65.4  2222.8    81.7  2212.3   114.4 2195.79
   150.4  2179.5   189.6  2164.8   212.5  2156.9   228.9 2155.07     242 2150.88
   268.1 2147.14   277.9 2148.22   297.5 2146.76   304.1 2144.98   310.6 2141.67
   317.2 2139.91   330.2 2139.78   359.6 2141.35   467.5 2143.68   506.8  2142.3
   519.9 2140.24   559.1 2143.42   575.4 2146.47   604.9 2160.03   634.3 2171.28
   660.4 2180.04   673.5 2183.31     703 2185.43   729.1 2185.93     801 2183.88
#Mann= 3 ,-1 , 0
       0      .1       0   310.6    .045       0   359.6      .1       0
Bank Sta=310.6,359.6
XS Rating Curve= 0 ,0
Exp/Cntr=0.3,0.1

Type RM Length L Ch R = 1 ,40397   ,697.9,684,638.2
XS GIS Cut Line= 3
     2128175.975      225984.061     2128375.409      226132.608
     2128999.648      226146.771
#Sta/Elev= 30
       0 2237.88    78.5 2214.91    88.4 2213.47   127.6 2202.58   157.1 2192.73
     180 2187.45   199.6 2182.03   212.7 2177.28   255.2 2158.43   274.8 2141.52
   284.6  2137.5   304.2 2137.12   323.9 2137.51   340.2 2141.01   353.3 2142.27
   389.2 2141.98   428.5 2140.89   444.8  2138.5   461.2 2139.97   493.9 2138.01
   523.3 2140.84   565.8 2140.21   614.8 2142.06   663.8 2141.99   706.4  2152.9
   722.7 2158.73   742.3  2163.2   778.3  2166.7   801.2 2166.57   873.1 2170.44
#Mann= 5 ,-1 , 0
       0      .1       0     180     .12       0   274.8    .045       0
   340.2     .12       0  408.68      .1       0
Bank Sta=274.8,340.2
XS Rating Curve= 0 ,0
Exp/Cntr=0.3,0.1

Type RM Length L Ch R = 1 ,39713   ,442.9,416.6,385
XS GIS Cut Line= 3
     2128532.808      226829.388     2128667.076      226625.663
       2129100.1      226304.052
#Sta/Elev= 30
       0 2237.12    16.3 2236.52    45.6  2232.6   100.8 2216.62   130.1 2205.21
   139.9 2203.67   169.2 2191.04   198.4  2182.8   214.7    2176   260.3 2154.03
     280 2138.76   289.8 2134.63   322.4 2133.18   335.5 2135.19   368.2 2135.09
   391.1 2132.61   417.2 2133.64   423.8 2136.28   433.6 2137.92   446.7 2138.28
   557.8 2132.96   574.2 2136.28     597  2137.6   616.7 2140.95   646.1 2153.58
   659.2 2157.95   678.8 2159.07   698.4 2162.48     718 2164.25   783.4 2177.36
#Mann= 7 ,-1 , 0
       0      .1       0      70     .08       0     170     .05       0
     190     .08       0  323.99      .1       0   368.2    .045       0
   423.8      .1       0
Bank Sta=368.2,423.8
XS Rating Curve= 0 ,0
Exp/Cntr=0.3,0.1

Type RM Length L Ch R = 1 ,39296   ,170.5,167.7,157.2
XS GIS Cut Line= 3
2129085.87294527227007.6442739782129136.41766916226546.540401275
     2129222.631226377.481616451
#Sta/Elev= 30
       0 2218.25    19.6 2215.64    32.7 2212.79    49.1 2210.81    98.1 2194.57
   104.7 2191.41   111.2 2186.12   117.7 2181.73   173.3 2155.76   196.2 2146.79
   219.1 2140.26   264.9 2136.01     278 2131.14   287.8 2128.93   304.2 2128.31
   310.7 2128.66   323.8 2131.25   336.9 2131.88   359.8 2130.75     399 2130.76
   412.1 2130.32   421.9 2129.15   431.7 2129.87   444.8 2132.25   477.5 2148.51
   493.8 2154.56   523.3 2161.81     556 2171.92   598.5 2180.03   624.7  2182.3
#Mann= 6 ,-1 , 0
       0    .035       0      40      .1       0     278    .045       0
   323.8      .1       0     340     .12       0     440      .1       0
Bank Sta=278,323.8
XS Rating Curve= 0 ,0
Exp/Cntr=0.3,0.1

Type RM Length L Ch R = 1 ,39129   ,330.6,358,370.8
XS GIS Cut Line= 3
2129303.93002518227054.2582638682129267.66446357226512.001771166
2129279.75298411226391.116565787
#Sta/Elev= 30
       0  2214.3    10.5 2212.55    36.8 2205.06    76.3 2190.99   102.6 2180.04
     119 2172.54   158.5 2156.98     198 2145.56   227.5 2135.91   246.7 2133.04
   293.3 2130.55   319.6 2127.73   352.5 2127.39     370 2127.77     392 2129.89
   428.1 2129.63     438 2131.02   441.7  2130.8   451.1 2128.33   457.7 2127.93
   477.4 2130.91     481  2131.9     507 2147.95   516.9  2153.1   539.5 2162.03
   564.4 2170.01   589.4 2176.27   606.8 2179.09   628.9 2181.91     665  2184.8
#Mann= 7 ,-1 , 0
       0      .1       0      90     .12       0     190      .1       0
     280     .12       0   319.6    .045       0     370     .12       0
     480      .1       0
Bank Sta=319.6,370
XS Rating Curve= 0 ,0
Exp/Cntr(USF)=0,0
Exp/Cntr=0.3,0.1

Type RM Length L Ch R = 1 ,38770   ,356.2,381.8,400.8
XS GIS Cut Line= 2
     2129438.097      227051.071     2129680.965      226455.524
#Sta/Elev= 30
       0 2190.25    16.3  2181.2    29.4 2178.92    32.6 2177.42    45.7  2169.9
   107.7  2139.7   127.3 2131.32   137.1 2129.22   156.7    2129   166.5 2129.98
   195.9 2127.01   212.2 2127.78   225.3 2130.12   280.8  2129.8   306.9 2127.32
   326.5 2127.72   346.1 2126.58   372.2 2127.68   401.6 2130.54   434.2 2126.14
   470.1 2123.92   489.7 2124.36   496.2 2127.22   509.3 2136.07   535.4  2147.8
   561.5 2165.26   581.1  2175.3   607.2  2185.5   630.1 2190.86   643.2 2192.63
#Mann= 3 ,-1 , 0
       0      .1       0   434.2    .045       0   496.2      .1       0
Bank Sta=434.2,496.2
XS Rating Curve= 0 ,0
Exp/Cntr=0.3,0.1

Type RM Length L Ch R = 1 ,38389   ,465.2,500,521.5
XS GIS Cut Line= 3
     2129550.755      227114.142     2129915.329      226841.216
     2130199.195      226640.136
#Sta/Elev= 30
       0 2192.32    32.8 2178.66    55.7 2166.37   114.7 2137.35     131 2127.54
   173.6 2122.24   196.6 2125.24   222.8 2126.26   255.6 2125.75   271.9    2123
   288.3 2123.62   321.1 2127.17   350.6 2126.37   422.6 2126.87   445.6 2122.62
   455.4 2122.28   468.4 2122.44   481.4  2126.7   523.7  2148.3   533.4  2150.8
   543.2 2157.47     566 2168.08   595.2 2184.34     618 2191.29   650.5 2204.43
   660.2 2206.02   712.2 2222.55     748 2231.18     761 2237.06   803.3 2261.17
#Mann= 5 ,-1 , 0
       0      .1       0   422.6    .045       0   481.4     .12       0
  575.41      .1       0  745.41     .12       0
Bank Sta=422.6,481.4
XS Rating Curve= 0 ,0
Exp/Cntr=0.3,0.1

Type RM Length L Ch R = 1 ,37889   ,192.3,194.1,194.4
XS GIS Cut Line= 3
     2129605.771      227224.841     2130178.777      227247.251
     2130505.179      227267.652
#Sta/Elev= 30
       0 2199.42      59 2178.35    88.5 2164.67   124.5  2144.3   140.9 2129.13
   147.5 2124.49   157.3 2121.66   173.7 2120.99   183.5    2119   199.9 2122.43
   216.3  2123.1   232.6 2120.45   314.6 2123.22   376.8 2121.54   416.2 2121.72
   435.8 2123.42   534.1 2123.62   553.8 2120.18   576.7 2119.72   596.3  2123.8
   612.7 2134.04   655.2 2151.27     665 2156.46   684.6 2162.12   723.9 2170.36
     737 2176.16   746.8 2177.05   795.8 2197.25   841.6 2214.31   900.5 2231.95
#Mann= 6 ,-1 , 0
       0     .05       0      10      .1       0   534.1    .045       0
   596.3      .1       0  603.44     .12       0  703.44      .1       0
Bank Sta=534.1,596.3
XS Rating Curve= 0 ,0
Exp/Cntr=0.3,0.1

Type RM Length L Ch R = 1 ,37695   ,337.6,376.3,392.6
XS GIS Cut Line= 2
 2129637.8913601 227394.796848162130444.48614654227462.325714002
#Sta/Elev= 30
       0  2200.1    34.1 2196.58    53.8 2192.34    96.6 2177.15   116.4 2167.68
   139.4 2154.19   148.6 2145.48     159 2132.67   175.6 2119.89   182.2 2117.16
   192.1 2116.92   208.6 2120.63   238.2 2117.38   264.5 2122.19   313.9 2120.67
   346.9 2122.02   369.9 2117.71   392.9 2121.12   469.42121.528   498.3 2118.85
   530.72119.328   550.6 2126.95   583.9 2136.64   623.9 2144.43   656.3 2153.54
   715.6 2175.41   761.7 2196.48   774.9 2198.88   781.4 2203.29   809.4 2216.33
#Mann= 7 ,-1 , 0
       0    .035       0      80      .1       0     370     .12       0
   469.4    .045       0   530.7      .1       0     570     .12       0
     670      .1       0
Bank Sta=469.4,530.7
XS Rating Curve= 0 ,0
Exp/Cntr(USF)=0,0
Exp/Cntr=0.3,0.1

Type RM Length L Ch R = 1 ,37318   ,169.6,160.7,153.7
XS GIS Cut Line= 2
     2129625.409      227410.386     2130239.993      227806.219
#Sta/Elev= 30
       0 2199.97    27.9 2198.21    62.1 2194.63    86.5 2189.57   117.3 2178.82
   128.8 2172.97   148.9 2160.99   169.5 2145.45   190.9 2132.15   199.6 2125.72
   207.4 2118.53   209.8 2117.32   221.7 2115.58   238.3 2115.14   252.42117.242
   304.8 2118.37   324.5 2120.53   433.8 2119.46   468.1 2121.56   506.6 2129.69
     516 2130.86   546.9 2138.45   558.7 2139.79   589.9 2146.43   619.5 2157.74
   636.7    2163   644.5 2164.26   660.1 2171.85   704.4  2187.9     731 2199.69
#Mann= 4 ,-1 , 0
       0    .035       0     100      .1       0   209.8    .045       0
   252.4      .1       0
Bank Sta=209.8,252.4
XS Rating Curve= 0 ,0
Exp/Cntr=0.3,0.1

Type RM Length L Ch R = 1 ,37158   ,364.8,404,432
XS GIS Cut Line= 2
2129619.13334181227638.6510859222130226.89313438227833.734476131
#Sta/Elev= 30
       0 2150.97      15 2148.42    93.3 2132.44   113.9 2125.82   124.3 2123.39
   138.1 2117.27     145 2115.57     176 2115.07   182.62115.537   193.2 2116.31
   227.7 2116.25   241.4 2118.31   270.6 2119.74   283.7  2119.3   303.5 2120.07
   324.1 2118.33   358.6 2117.99   380.2 2118.81   393.2 2120.67   403.6 2124.64
     431 2132.59   475.7 2149.36     501 2158.18   511.8 2161.06   539.3 2171.29
     555 2173.76   561.9 2177.19   589.5 2186.12   614.9 2196.83   638.3 2205.61
#Mann= 3 ,-1 , 0
       0      .1       0   138.1    .045       0   182.6      .1       0
Bank Sta=138.1,182.6
XS Rating Curve= 0 ,0
Exp/Cntr(USF)=0,0
Exp/Cntr=0.3,0.1

Type RM Length L Ch R = 1 ,36753   ,252.7,255.7,256.8
XS GIS Cut Line= 2
2129611.63013449227657.4091042112129840.47795762228373.965402863
#Sta/Elev= 30
       0 2146.69    48.1 2137.59      86 2122.44     117 2115.84   137.6    2119
   170.5 2118.21   186.2 2116.13   216.8 2119.27   261.6 2116.99   298.4 2118.91
   371.5 2116.39     395 2114.81   405.2  2112.4   430.4 2109.66   447.6 2109.93
   454.5 2111.82   457.32113.637   461.4 2117.72   478.3 2137.71   492.4 2147.24
   522.9 2163.52   547.5 2174.94     596 2203.23   612.9 2210.57   629.9 2219.65
   650.7 2227.14   672.4 2232.27     730 2240.89   739.6 2243.65   752.2 2243.69
#Mann= 6 ,-1 , 0
       0      .1       0     320     .12       0   405.2    .045       0
   457.3     .12       0     630      .1       0     730     .05       0
Bank Sta=405.2,457.3
XS Rating Curve= 0 ,0
Exp/Cntr(USF)=0,0
Exp/Cntr=0.3,0.1

Type RM Length L Ch R = 1 ,36498   ,285.9,289.5,291.5
XS GIS Cut Line= 2
     2129404.468      227765.902      2129586.72      228470.748
#Sta/Elev= 30
       0 2140.38    26.2  2136.5    52.5 2131.12    62.3 2127.48    88.5  2114.9
   101.7 2111.52   114.8 2111.33   127.9 2114.51     164 2116.78     200 2116.67
   219.7 2116.43     246    2114   265.6 2115.96   318.1 2113.99   341.1 2114.36
   354.2 2113.71   370.6 2110.88   383.7    2111   400.1 2110.64   413.2 2108.95
   432.9 2109.08   439.4 2111.17   452.6 2125.85   455.8 2128.09   501.8 2150.47
   580.4 2191.35   623.1 2212.27   655.9 2223.58   711.6 2239.36     728  2241.4
#Mann= 6 ,-1 , 0
       0      .1       0     100     .12       0     200      .1       0
     300     .12       0   383.7    .045       0   439.4      .1       0
Bank Sta=383.7,439.4
XS Rating Curve= 0 ,0
Exp/Cntr=0.3,0.1

Type RM Length L Ch R = 1 ,36208   ,319.5,319.6,317.9
XS GIS Cut Line= 3
     2129158.437      227822.597     2129217.695      228181.518
     2129284.241      228540.403
#Sta/Elev= 30
       0 2150.67      36 2143.77    52.4 2137.45    65.6 2136.98    78.7 2133.86
   111.4 2124.44   121.3 2122.77   144.2 2113.35   163.9 2108.46   209.8 2112.97
   249.1 2110.07   268.7 2111.54   314.6 2112.17   321.2 2111.63   334.3 2107.29
     354 2110.47   380.1 2109.85   399.6 2106.16   406.2 2105.82   432.2 2106.68
     442 2110.68     455 2119.37   500.7 2143.62   533.2 2162.45   549.5 2170.79
   569.1  2179.4   604.9 2192.42   637.5 2199.71   696.2 2210.73   728.8 2219.22
#Mann= 3 ,-1 , 0
       0      .1       0   380.1    .045       0     442      .1       0
Bank Sta=380.1,442
XS Rating Curve= 0 ,0
Exp/Cntr=0.3,0.1

Type RM Length L Ch R = 1 ,35889   ,333.5,328.6,322.1
XS GIS Cut Line= 3
     2128840.197      227932.049     2128914.437      228288.398
     2128988.676      228644.747
#Sta/Elev= 30
       0 2171.84    13.1 2163.76    19.7 2160.57    65.6  2143.6    78.7 2138.09
    88.5 2135.36   150.8  2108.9   167.2 2103.57   170.5 2103.33   183.6 2105.37
   216.4 2106.73   239.4 2105.92   311.5 2107.95   331.2 2106.66   344.3 2104.26
   377.1 2103.64     387 2104.34   393.5 2107.13   413.2 2121.11   455.8 2143.22
   475.5 2150.96   501.7  2159.9   541.1 2174.84   583.7 2189.88   613.2 2198.12
   636.2 2205.48     669 2213.65   682.1 2217.82   714.9 2226.41     728  2231.1
#Mann= 3 ,-1 , 0
       0      .1       0   331.2    .045       0   393.5      .1       0
Bank Sta=331.2,393.5
XS Rating Curve= 0 ,0
Exp/Cntr=0.3,0.1

Type RM Length L Ch R = 1 ,35560   ,420.4,421.4,405.3
XS GIS Cut Line= 3
     2128465.316      228014.737     2128592.349      228355.581
     2128717.168      228698.962
#Sta/Elev= 30
       0 2184.84    49.2 2157.66    88.5 2140.73     118 2121.76   147.5 2107.65
   180.2  2100.6   196.6 2103.25   216.3 2104.57   245.8 2103.06   255.6 2100.45
   275.3 2103.46   321.2 2102.12   334.2 2103.41   363.8 2103.16   393.1 2100.56
   412.7 2100.96   419.2 2103.41   432.2 2109.96   451.8  2125.2   458.4 2132.02
   464.9 2142.59   468.1 2146.36   494.2 2166.46   513.8 2185.15   526.9 2191.36
   569.3 2204.06   595.4 2213.27   614.9  2217.7   670.4 2226.14   729.1 2230.58
#Mann= 3 ,-1 , 0
       0      .1       0   363.8    .045       0   419.2      .1       0
Bank Sta=363.8,419.2
XS Rating Curve= 0 ,0
Exp/Cntr=0.3,0.1

Type RM Length L Ch R = 1 ,35139   ,298.3,290.6,275.2
XS GIS Cut Line= 3
     2128018.696      228195.368     2128239.712      228469.745
     2128517.077      228804.232
#Sta/Elev= 30
       0 2200.02    26.1 2184.61    48.9 2169.24    71.8 2156.73   153.3 2106.36
   166.4 2100.27   176.2 2097.66   189.2 2097.42   238.1 2103.19     261 2099.06
   270.8 2099.83   293.6 2097.94   316.4 2100.75   329.5 2097.92   339.3 2096.76
   362.1 2096.81   371.9 2098.43   388.3 2100.91   391.5 2100.69   401.3  2097.1
   437.3 2098.65   453.6 2105.73   473.2 2111.92   512.4 2130.27   528.8 2135.43
   626.8 2154.62   682.3 2163.14   705.2 2168.38   737.8 2173.44   786.8 2184.03
#Mann= 3 ,-1 , 0
       0      .1       0   329.5    .045       0   371.9      .1       0
Bank Sta=329.5,371.9
XS Rating Curve= 0 ,0
Exp/Cntr=0.3,0.1

Type RM Length L Ch R = 1 ,34848   ,511.8,509.1,462.4
XS GIS Cut Line= 3
     2127712.215      228403.441      2127799.02       228511.08
      2128436.77      228891.409
#Sta/Elev= 30
       0 2199.47    19.3 2187.25    28.9 2178.81    54.7 2159.47    64.3 2157.03
    96.5 2138.03   128.6 2121.93   138.3 2119.75   164.4 2109.51   193.9  2095.5
   233.1 2100.33   347.6 2099.87     364 2098.32   383.6 2099.25     400 2097.43
   419.6 2098.59   429.4 2096.83   442.5 2094.96   507.9 2095.14   514.5 2097.13
   524.3 2099.56     557 2099.96   586.4 2112.71   602.8  2118.3   619.1 2121.34
   645.3 2124.66   753.2 2132.53     822 2140.27   854.7 2144.88   880.8 2152.68
#Mann= 5 ,-1 , 0
       0      .1       0  408.28     .12       0   429.4    .045       0
   514.5     .12       0  758.28      .1       0
Bank Sta=429.4,514.5
XS Rating Curve= 0 ,0
Exp/Cntr=0.3,0.1

Type RM Length L Ch R = 1 ,34339   ,545.5,511.4,442.9
XS GIS Cut Line= 3
     2127476.104      229021.497     2127726.104      228958.997
     2128417.076      228913.858
#Sta/Elev= 30
       0  2249.9    45.7 2224.65    58.7 2214.42    71.8 2211.84    91.3 2199.31
   117.4 2185.53   156.6 2166.31   163.1 2165.18   228.3 2131.09   238.1 2124.65
   280.6 2104.12   293.6 2094.82   300.2 2090.98   313.2 2090.35   329.6 2090.58
   365.5 2094.18   401.4 2092.28     421 2095.88   447.1 2095.12   463.5 2097.18
   505.9 2098.06   545.1 2096.18   603.9 2096.51   623.5 2092.61   649.6 2095.37
   669.2 2094.63   760.7 2110.13   832.6 2117.36   927.3 2136.44   950.1 2143.11
#Mann= 6 ,-1 , 0
       0     .08       0      70      .1       0   293.6    .045       0
   365.5      .1       0  667.69     .12       0  767.69      .1       0
Bank Sta=293.6,365.5
XS Rating Curve= 0 ,0
Exp/Cntr=0.3,0.1

Type RM Length L Ch R = 1 ,33828   ,331.6,364.2,407.7
XS GIS Cut Line= 4
2127644.20128661229410.2157012382128069.72103111229319.369524645
     2128229.576      228972.886      2128424.02      228952.052
#Sta/Elev= 30
       0 2169.58    20.2 2164.16    53.4 2157.36   171.2 2137.67   261.8 2130.29
   308.7 2122.41   342.3 2119.19   422.8 2115.71   435.1 2113.76   448.1 2114.53
   459.7 2112.95   467.1 2110.01     477 2100.22   484.4  2095.4   495.1 2092.34
   526.42088.455   545.7 2085.64   578.4 2085.45   585.8 2085.99   592.6 2088.28
   602.2 2091.77   614.4 2094.11   664.9 2092.89   677.3 2094.78   793.5 2097.17
   828.6 2104.95   907.8  2115.1   957.3 2126.52   970.5 2131.06  1012.2 2141.31
#Mann= 8 ,-1 , 0
       0      .1       0     370     .12       0     400      .1       0
   526.4    .045       0   592.6     .12       0  635.11      .1       0
  745.11     .12       0  826.69      .1       0
Bank Sta=526.4,592.6
XS Rating Curve= 0 ,0
Exp/Cntr=0.3,0.1
